HEC-RAS study P100-00-00.prj: P100-00-00

--- P100-00-00.p02 (plan) ---

Plan Title=Effective Floodway 2020
Program Version=5.07
Short Identifier=Effective FW 2020
Geom File=g01
Flow File=f02
Subcritical Flow
K Sum by GR= 0
Std Step Tol= 0.01
Critical Tol= 0.01
Num of Std Step Trials= 20
Max Error Tol= 0.3
Flow Tol Ratio= 0.001
Split Flow NTrial= 30
Split Flow Tol= 0.02
Split Flow Ratio= 0.02
Log Output Level= 0
Friction Slope Method= 1
Unsteady Friction Slope Method= 2
Unsteady Bridges Friction Slope Method= 1
Parabolic Critical Depth
Global Vel Dist= 0 , 0 , 0
Global Log Level= 0
CheckData=True
Encroach Param= 0 ,0,0, 5
Encroach River=P100-00-00
Encroach Reach=P100-00-00_0010
Encroach Node=228675.4
       1    4976  5020.3       0       0       0       0       0       0
       1    4976  5020.3
Encroach Node=228484.7
       1    4976  5020.3       0       0       0       0       0       0
       1    4976  5020.3
Encroach Node=228436.2
       1  4980.1  5022.4       0       0       0       0       0       0
       1  4980.1  5022.4
Encroach Node=228380.9
       1    4972    5050       0       0       0       0       0       0
       1    4972    5050
Encroach Node=228325.7
       1  4980.1  5020.6       0       0       0       0       0       0
       1  4980.1  5020.6
Encroach Node=227921.0
       1  4965.4  5032.9       0       0       0       0       0       0
       1  4965.4  5032.9
Encroach Node=227282.4
       1    4965  5032.9       0       0       0       0       0       0
       1    4965  5032.9
Encroach Node=226694.3
       1    4962    5045       0       0       0       0       0       0
       1    4962    5045
Encroach Node=226400.3
       1    4941    5046       0       0       0       0       0       0
       1    4941    5046
Encroach Node=226342.8
       1    4941    5046       0       0       0       0       0       0
       1    4941    5046
Encroach Node=226285.3
       1    4941    5046       0       0       0       0       0       0
       1    4941    5046
Encroach Node=225939.1
       1  4954.6  5036.7       0       0       0       0       0       0
       1  4954.6  5036.7
Encroach Node=225480.0
       1  4954.6  5036.7       0       0       0       0       0       0
       1  4954.6  5036.7
Encroach Node=225142.8
       1  4954.6  5036.7       0       0       0       0       0       0
       1  4954.6  5036.7
Encroach Node=225131.3
       1  4954.6  5036.7       0       0       0       0       0       0
       1  4954.6  5036.7
Encroach Node=225119.8
       1  4954.6  5036.7       0       0       0       0       0       0
       1  4954.6  5036.7
Encroach Node=224949.2
       1    4965    5033       0       0       0       0       0       0
       1    4965    5033
Encroach Node=224889.7
       1    4965    5033       0       0       0       0       0       0
       1    4965    5033
Encroach Node=224830.2
       1    4965    5033       0       0       0       0       0       0
       1    4965    5033
Encroach Node=224308.4
       1  4954.4  5049.3       0       0       0       0       0       0
       1  4954.4  5049.3
Encroach Node=223997.9
       1  4954.4  5049.3       0       0       0       0       0       0
       1  4954.4  5049.3
Encroach Node=223061.5
       1  4956.8  5053.3       0       0       0       0       0       0
       1  4956.8  5053.3
Encroach Node=221964.2
       1    4960  5049.3       0       0       0       0       0       0
       1    4960  5049.3
Encroach Node=221230.4
       1  4982.7  5058.4       0       0       0       0       0       0
       1  4982.7  5058.4
Encroach Node=220984.2
       1  4982.7  5058.4       0       0       0       0       0       0
       1  4982.7  5058.4
Encroach Node=220925.7
       1  4982.7  5058.4       0       0       0       0       0       0
       1  4982.7  5058.4
Encroach Node=220867.3
       1  4982.7  5058.4       0       0       0       0       0       0
       1  4982.7  5058.4
Encroach Node=220631.9
       1  4933.3  5044.4       0       0       0       0       0       0
       1  4933.3  5044.4
Encroach Node=220575.9
       1  4933.3  5044.4       0       0       0       0       0       0
       1  4933.3  5044.4
Encroach Node=220519.9
       1  4933.3  5044.4       0       0       0       0       0       0
       1  4933.3  5044.4
Encroach Node=220257.4
       1  4952.3  5041.8       0       0       0       0       0       0
       1  4952.3  5041.8
Encroach Node=219998.9
       1  4952.3  5041.8       0       0       0       0       0       0
       1  4952.3  5041.8
Encroach Node=219744.4
       1 4874.51  5041.8       0       0       0       0       0       0
       1 4874.51  5041.8
Encroach Node=219716.4
       1 4874.51  5041.8       0       0       0       0       0       0
       1 4874.51  5041.8
Encroach Node=219688.4
       1 4874.51  5041.8       0       0       0       0       0       0
       1 4874.51  5041.8
Encroach Node=219073.4
       1  4976.7  5024.6       0       0       0       0       0       0
       1  4976.7  5024.6
Encroach Node=218243.5
       1    4800    5250       0       0       0       0       0       0
       1    4800    5250
Encroach Node=218103.7
       1    4830    5400       0       0       0       0       0       0
       1    4830    5400
Encroach Node=218075.2
       1    4830    5400       0       0       0       0       0       0
       1    4830    5400
Encroach Node=218046.7
       1    4830    5400       0       0       0       0       0       0
       1    4830    5400
Encroach Node=217461.8
       1    4750    5400       0       0       0       0       0       0
       1    4750    5400
Encroach Node=217089.5
       1    4725    5650       0       0       0       0       0       0
       1    4725    5650
Encroach Node=216460.9
       1    4700    5040       0       0       0       0       0       0
       1    4700    5040
Encroach Node=215936.4
       1  4975.3  5021.6       0       0       0       0       0       0
       1  4975.3  5021.6
Encroach Node=215326.4
       1    4954    5060       0       0       0       0       0       0
       1    4954    5060
Encroach Node=214983.1
       1    4913    5085       0       0       0       0       0       0
       1    4913    5085
Encroach Node=214927.1
       1    4913    5085       0       0       0       0       0       0
       1    4913    5085
Encroach Node=214871.1
       1    4913    5085       0       0       0       0       0       0
       1    4913    5085
Encroach Node=213673.1
       1    4900    5090       0       0       0       0       0       0
       1    4900    5090
Encroach Node=212608.8
       1    4900    5090       0       0       0       0       0       0
       1    4900    5090
Encroach Node=212060.6
       1    4850    5100       0       0       0       0       0       0
       1    4850    5100
Encroach Node=211630.6
       1    4900    5100       0       0       0       0       0       0
       1    4900    5100
Encroach Node=211602.6
       1    4900    5100       0       0       0       0       0       0
       1    4900    5100
Encroach Node=211574.6
       1    4900    5100       0       0       0       0       0       0
       1    4900    5100
Encroach Node=211066.9
       1    4900    5089       0       0       0       0       0       0
       1    4900    5089
Encroach Node=210776.9
       1    4900    5089       0       0       0       0       0       0
       1    4900    5089
Encroach Node=210486.9
       1    4900    5089       0       0       0       0       0       0
       1    4900    5089
Encroach Node=210022.7
       1    4870    5100       0       0       0       0       0       0
       1    4870    5100
Encroach Node=209411.0
       1    4903    5063       0       0       0       0       0       0
       1    4903    5063
Encroach Node=209391.0
       1    4903    5063       0       0       0       0       0       0
       1    4903    5063
Encroach Node=209371.0
       1    4903    5063       0       0       0       0       0       0
       1    4903    5063
Encroach Node=209281.4
       1    4903    5063       0       0       0       0       0       0
       1    4903    5063
Encroach Node=209256.4
       1    4903    5063       0       0       0       0       0       0
       1    4903    5063
Encroach Node=209231.4
       1    4930    5063       0       0       0       0       0       0
       1    4930    5063
Encroach Node=208303.8
       1    4900    5100       0       0       0       0       0       0
       1    4900    5100
Encroach Node=207557.1
       1    4850    5100       0       0       0       0       0       0
       1    4850    5100
Encroach Node=206854.1
       1    4900    5100       0       0       0       0       0       0
       1    4900    5100
Encroach Node=206174.0
       1    4920    5076       0       0       0       0       0       0
       1    4920    5076
Encroach Node=206145.5
       1    4920    5076       0       0       0       0       0       0
       1    4920    5076
Encroach Node=206117.0
       1    4920    5076       0       0       0       0       0       0
       1    4920    5076
Encroach Node=205188.9
       1    4800    5200       0       0       0       0       0       0
       1    4800    5200
Encroach Node=204744.1
       1    4800    5200       0       0       0       0       0       0
       1    4800    5200
Encroach Node=203825.7
       1    4800    5225       0       0       0       0       0       0
       1    4800    5225
Encroach Node=202904.2
       1    4775    5200       0       0       0       0       0       0
       1    4775    5200
Encroach Node=201967.0
       1    4800    5200       0       0       0       0       0       0
       1    4800    5200
Encroach Node=201733.0
       1    4795    5285       0       0       0       0       0       0
       1    4795    5285
Encroach Node=200823.6
       1    4750    5300       0       0       0       0       0       0
       1    4750    5300
Encroach Node=200063.8
       1    4700    5150       0       0       0       0       0       0
       1    4700    5150
Encroach Node=199501.1
       1    4840    5150       0       0       0       0       0       0
       1    4840    5150
Encroach Node=198785.6
       1  4909.7  5078.8       0       0       0       0       0       0
       1  4909.7  5078.8
Encroach Node=198726.8
       1  4909.7  5078.8       0       0       0       0       0       0
       1  4909.7  5078.8
Encroach Node=198668.1
       1  4909.7  5078.8       0       0       0       0       0       0
       1  4909.7  5078.8
Encroach Node=198192.4
       1  4950.9  5088.6       0       0       0       0       0       0
       1  4950.9  5088.6
Encroach Node=197172.9
       1  4937.5  5078.9       0       0       0       0       0       0
       1  4937.5  5078.9
Encroach Node=196097.0
       1    4935    5090       0       0       0       0       0       0
       1    4935    5090
Encroach Node=194928.6
       1    4755    5145       0       0       0       0       0       0
       1    4755    5145
Encroach Node=194146.5
       1    4920    5550       0       0       0       0       0       0
       1    4920    5550
Encroach Node=193896.3
       1    4900    5550       0       0       0       0       0       0
       1    4900    5550
Encroach Node=193838.8
       1    4900    5550       0       0       0       0       0       0
       1    4900    5550
Encroach Node=193781.3
       1    4900    5550       0       0       0       0       0       0
       1    4900    5550
Encroach Node=192935.6
       1  4952.4    5480       0       0       0       0       0       0
       1  4952.4    5480
Encroach Node=191836.0
       1    4880  5077.3       0       0       0       0       0       0
       1    4880  5077.3
Encroach Node=191278.6
       1    4916  5126.5       0       0       0       0       0       0
       1    4916  5126.5
Encroach Node=190860.1
       1 4944.25 5109.35       0       0       0       0       0       0
       1 4944.25 5109.35
Encroach Node=190848.1
       1 4944.25 5109.35       0       0       0       0       0       0
       1 4944.25 5109.35
Encroach Node=190836.1
       1 4944.25 5109.35       0       0       0       0       0       0
       1 4944.25 5109.35
Encroach Node=190772.0
       1 4923.41 5089.54       0       0       0       0       0       0
       1 4923.41 5089.54
Encroach Node=190739.5
       1 4923.41 5089.54       0       0       0       0       0       0
       1 4923.41 5089.54
Encroach Node=190707.0
       1 4923.41 5089.54       0       0       0       0       0       0
       1 4923.41 5089.54
Encroach Node=189685.2
       1  4931.6    5100       0       0       0       0       0       0
       1  4931.6    5100
Encroach Node=188681.0
       1  4928.4  5090.5       0       0       0       0       0       0
       1  4928.4  5090.5
Encroach Node=187593.9
       1  4907.7  5078.9       0       0       0       0       0       0
       1  4907.7  5078.9
Encroach Node=187053.5
       1  4888.8  5091.6       0       0       0       0       0       0
       1  4888.8  5091.6
Encroach Node=186609.7
       1  4929.4  5091.6       0       0       0       0       0       0
       1  4929.4  5091.6
Encroach Node=186581.7
       1  4929.4  5091.6       0       0       0       0       0       0
       1  4929.4  5091.6
Encroach Node=186553.7
       1  4929.4  5091.6       0       0       0       0       0       0
       1  4929.4  5091.6
Encroach Node=186025.8
       1  4938.6  5100.8       0       0       0       0       0       0
       1  4938.6  5100.8
Encroach Node=185578.7
       1  4938.6  5100.8       0       0       0       0       0       0
       1  4938.6  5100.8
Encroach Node=184592.5
       1 4917.15 5136.68       0       0       0       0       0       0
       1 4917.15 5136.68
Encroach Node=184557.5
       1 4917.15 5136.68       0       0       0       0       0       0
       1 4917.15 5136.68
Encroach Node=184522.5
       1 4917.15 5136.68       0       0       0       0       0       0
       1 4917.15 5136.68
Encroach Node=184421.0
       1  4840.6    5450       0       0       0       0       0       0
       1  4840.6    5450
Encroach Node=184343.0
       1  4840.6    5785       0       0       0       0       0       0
       1  4840.6    5785
Encroach Node=184265.0
       1 4840.46    5149       0       0       0       0       0       0
       1 4840.46    5149
Encroach Node=184132.4
       1 4894.43 5144.76       0       0       0       0       0       0
       1 4894.43 5144.76
Encroach Node=184097.4
       1 4894.43 5144.76       0       0       0       0       0       0
       1 4894.43 5144.76
Encroach Node=184062.4
       1 4894.43 5144.76       0       0       0       0       0       0
       1 4894.43 5144.76
Encroach Node=183348.2
       1    4885  5055.4       0       0       0       0       0       0
       1    4885  5055.4
Encroach Node=181918.8
       1 4881.22 5090.56       0       0       0       0       0       0
       1 4881.22 5090.56
Encroach Node=181883.8
       1 4881.22 5090.56       0       0       0       0       0       0
       1 4881.22 5090.56
Encroach Node=181848.8
       1 4881.22 5090.56       0       0       0       0       0       0
       1 4881.22 5090.56
Encroach Node=181739.5
       1 4877.63 5121.47       0       0       0       0       0       0
       1 4877.63 5121.47
Encroach Node=181661.5
       1 4877.63 5121.47       0       0       0       0       0       0
       1 4877.63 5121.47
Encroach Node=181583.5
       1 4877.63 5121.47       0       0       0       0       0       0
       1 4877.63 5121.47
Encroach Node=181519.5
       1 4878.53 5100.42       0       0       0       0       0       0
       1 4878.53 5100.42
Encroach Node=181484.5
       1 4878.53 5100.42       0       0       0       0       0       0
       1 4878.53 5100.42
Encroach Node=181449.5
       1 4878.53 5100.42       0       0       0       0       0       0
       1 4878.53 5100.42
Encroach Node=180957.6
       1  4931.9  5058.9       0       0       0       0       0       0
       1  4931.9  5058.9
Encroach Node=179921.2
       1  4929.7  5085.1       0       0       0       0       0       0
       1  4929.7  5085.1
Encroach Node=179126.0
       1  4911.6  5069.1       0       0       0       0       0       0
       1  4911.6  5069.1
Encroach Node=178828.2
       1  4911.6  5084.4       0       0       0       0       0       0
       1  4911.6  5084.4
Encroach Node=178803.2
       1  4911.6  5084.4       0       0       0       0       0       0
       1  4911.6  5084.4
Encroach Node=178778.2
       1  4911.6  5084.4       0       0       0       0       0       0
       1  4911.6  5084.4
Encroach Node=178661.5
       1  4911.3  5081.7       0       0       0       0       0       0
       1  4916.3  5081.7
Encroach Node=178636.5
       1  4911.3  5081.7       0       0       0       0       0       0
       1  4916.3  5081.7
Encroach Node=178611.5
       1  4911.3  5081.7       0       0       0       0       0       0
       1  4916.3  5081.7
Encroach Node=177406.7
       1  4940.9  5101.8       0       0       0       0       0       0
       1  4940.9  5101.8
Encroach Node=176342.1
       1    4888  5053.6       0       0       0       0       0       0
       1    4888  5053.6
Encroach Node=175998.8
       1    4920    5340       0       0       0       0       0       0
       1    4920    5340
Encroach Node=175549.5
       1    4830    5270       0       0       0       0       0       0
       1    4830    5270
Encroach Node=175538.0
       1    4830    5270       0       0       0       0       0       0
       1    4830    5270
Encroach Node=175525.6
       1    4830    5270       0       0       0       0       0       0
       1    4830    5270
Encroach Node=175483.1
       1    4710    5456       0       0       0       0       0       0
       1    4830    5270
Encroach Node=175440.6
       1    4830    5270       0       0       0       0       0       0
       1    4830    5270
Encroach Node=175354.9
       1  4825.7  5250.7       0       0       0       0       0       0
       0       0       0
Encroach Node=175300.3
       1    4830    5285       0       0       0       0       0       0
       0       0       0
Encroach Node=175203.7
       1    4820    5290       0       0       0       0       0       0
       0       0       0
Encroach Node=175146.3
       1  4845.1  5230.1       0       0       0       0       0       0
       0       0       0
Encroach Node=174932.7
       1    4800    5115       0       0       0       0       0       0
       0       0       0
Encroach Node=174086.8
       1    4850    5120       0       0       0       0       0       0
       1    4850    5120
Encroach Node=173023.1
       1    4840  5067.8       0       0       0       0       0       0
       1    4840  5067.8
Encroach Node=172472.6
       1    4910    5130       0       0       0       0       0       0
       1    4910    5130
Encroach Node=171583.6
       1    4865    5135       0       0       0       0       0       0
       1    4865    5135
Encroach Node=170916.5
       1    4850    5150       0       0       0       0       0       0
       1    4850    5150
Encroach Node=170549.0
       1    4830    5150       0       0       0       0       0       0
       1    4830    5150
Encroach Node=170266.6
       1    4795    5220       0       0       0       0       0       0
       1    4795    5220
Encroach Node=170232.1
       1    4795    5220       0       0       0       0       0       0
       1    4795    5220
Encroach Node=170197.6
       1    4795    5220       0       0       0       0       0       0
       1    4795    5220
Encroach Node=169760.8
       1    4780    5220       0       0       0       0       0       0
       1    4780    5220
Encroach Node=169319.2
       1    4625    5250       0       0       0       0       0       0
       1    4625    5250
Encroach Node=169305.2
       1    4625    5250       0       0       0       0       0       0
       1    4625    5250
Encroach Node=169291.2
       1    4625    5250       0       0       0       0       0       0
       1    4625    5250
Encroach Node=169017.5
       1    4725    5140       0       0       0       0       0       0
       1    4725    5140
Encroach Node=168762.1
       1    4800    5200       0       0       0       0       0       0
       1    4800    5200
Encroach Node=168734.1
       1    4800    5200       0       0       0       0       0       0
       1    4800    5200
Encroach Node=168706.1
       1    4800    5200       0       0       0       0       0       0
       1    4800    5200
Encroach Node=168680.5
       1    4876  5124.3       0       0       0       0       0       0
       1    4876  5124.3
Encroach Node=168562.9
       1    4876  5124.3       0       0       0       0       0       0
       1    4876  5124.3
Encroach Node=168445.4
       1    4876  5124.3       0       0       0       0       0       0
       1    4876  5124.3
Encroach Node=168426.4
       1    4876  5120.2       0       0       0       0       0       0
       1    4876  5120.2
Encroach Node=168398.4
       1    4876  5120.2       0       0       0       0       0       0
       1    4876  5120.2
Encroach Node=168370.4
       1    4876  5120.2       0       0       0       0       0       0
       1    4876  5120.2
Encroach Node=168052.4
       1    4500    5400       0       0       0       0       0       0
       1    4500    5400
Encroach Node=167711.6
       1    4200    5400       0       0       0       0       0       0
       1    4200    5400
Encroach Node=167685.1
       1    4200    5400       0       0       0       0       0       0
       1    4200    5400
Encroach Node=167658.6
       1    4200    5400       0       0       0       0       0       0
       1    4200    5400
Encroach Node=166814.8
       1    4050    5120       0       0       0       0       0       0
       1    4050    5120
Encroach Node=165731.4
       1    3950    5115       0       0       0       0       0       0
       1    3950    5115
Encroach Node=164812.5
       1    4120    5200       0       0       0       0       0       0
       1    4120    5200
Encroach Node=164153.5
       1    4125    5210       0       0       0       0       0       0
       1    4125    5210
Encroach Node=163691.0
       1    4250    5200       0       0       0       0       0       0
       1    4250    5200
Encroach Node=163641.0
       1    4250    5200       0       0       0       0       0       0
       1    4250    5200
Encroach Node=163591.0
       1    4250    5200       0       0       0       0       0       0
       1    4250    5200
Encroach Node=163254.1
       1    4290    5200       0       0       0       0       0       0
       1    4290    5200
Encroach Node=163020.2
       1 4283.86    5200       0       0       0       0       0       0
       1 4283.86    5200
Encroach Node=163006.2
       1 4283.86    5200       0       0       0       0       0       0
       1 4283.86    5200
Encroach Node=162992.2
       1 4283.86    5200       0       0       0       0       0       0
       1 4283.86    5200
Encroach Node=162338.1
       1    4250    5285       0       0       0       0       0       0
       1    4250    5285
Encroach Node=161801.4
       1    4045    5750       0       0       0       0       0       0
       1    4045    5750
Encroach Node=160657.9
       1    3700    5830       0       0       0       0       0       0
       1    3700    5830
Encroach Node=160192.5
       1    3500    5595       0       0       0       0       0       0
       1    3500    5595
Encroach Node=159787.1
       1    3300    5400       0       0       0       0       0       0
       1    3300    5400
Encroach Node=159734.6
       1    3300    5400       0       0       0       0       0       0
       1    3300    5400
Encroach Node=159682.1
       1    3500    5400       0       0       0       0       0       0
       1    3500    5400
Encroach Node=158963.8
       1    3490    5455       0       0       0       0       0       0
       1    3490    5455
Encroach Node=157981.7
       1    3715    5795       0       0       0       0       0       0
       1    3715    5795
Encroach Node=156861.1
       1    4315    7150       0       0       0       0       0       0
       1    4315    7150
Encroach Node=156281.6
       1    4510    6000       0       0       0       0       0       0
       1    4510    6000
Encroach Node=155841.8
       1    4525    6000       0       0       0       0       0       0
       1    4525    6000
Encroach Node=155786.8
       1    4525    6000       0       0       0       0       0       0
       1    4525    6000
Encroach Node=155731.8
       1    4525    6000       0       0       0       0       0       0
       1    4525    6000
Encroach Node=155378.8
       1    4862    9141       0       0       0       0       0       0
       1    4862    9141
Encroach Node=155355.8
       1    4862    9141       0       0       0       0       0       0
       1    4862    9141
Encroach Node=155332.8
       1    4862    9141       0       0       0       0       0       0
       1    4862    9141
Encroach Node=155312.4
       1    4862    9141       0       0       0       0       0       0
       1    4862    9141
Encroach Node=155283.9
       1    4862    9141       0       0       0       0       0       0
       1    4862    9141
Encroach Node=155255.4
       1    4862    9141       0       0       0       0       0       0
       1    4862    9141
Encroach Node=155248.9
       1    4862    9141       0       0       0       0       0       0
       1    4862    9141
Encroach Node=155189.1
       1    4862    9141       0       0       0       0       0       0
       1    4862    9141
Encroach Node=155129.3
       1    4862    9141       0       0       0       0       0       0
       1    4862    9141
Encroach Node=155110.5
       1    4862    9141       0       0       0       0       0       0
       1    4862    9141
Encroach Node=155085.5
       1    4862    9141       0       0       0       0       0       0
       1    4862    9141
Encroach Node=155060.5
       1    4862    9141       0       0       0       0       0       0
       1    4862    9141
Encroach Node=154008.5
       1    4300    5700       0       0       0       0       0       0
       1    4300    5700
Encroach Node=152906.6
       1    4800    6450       0       0       0       0       0       0
       1    4800    6450
Encroach Node=151806.5
       1    4850    6950       0       0       0       0       0       0
       1    4850    6950
Encroach Node=150830.2
       1    4600    7000       0       0       0       0       0       0
       1    4600    7000
Encroach Node=149842.1
       1    4775    6600       0       0       0       0       0       0
       1    4775    6600
Encroach Node=148819.5
       1    4600    6150       0       0       0       0       0       0
       1    4600    6150
Encroach Node=147831.4
       1    4780    5480       0       0       0       0       0       0
       1    4780    5480
Encroach Node=146526.5
       1    4430    5345       0       0       0       0       0       0
       1    4430    5345
Encroach Node=145462.0
       1    4450    5300       0       0       0       0       0       0
       1    4450    5300
Encroach Node=145018.0
       1    4450    5300       0       0       0       0       0       0
       1    4450    5300
Encroach Node=144651.8
       1    4400    5280       0       0       0       0       0       0
       1    4400    5280
Encroach Node=144624.3
       1    4400    5280       0       0       0       0       0       0
       1    4400    5280
Encroach Node=144596.8
       1    4400    5280       0       0       0       0       0       0
       1    4400    5280
Encroach Node=144556.0
       1    4400    5280       0       0       0       0       0       0
       1    4400    5280
Encroach Node=144545.0
       1    4400    5280       0       0       0       0       0       0
       1    4400    5280
Encroach Node=144534.0
       1    4400    5280       0       0       0       0       0       0
       1    4400    5280
Encroach Node=143348.1
       1    4050    5350       0       0       0       0       0       0
       1    4050    5350
Encroach Node=142602
       1    3940    5780       0       0       0       0       0       0
       0       0       0
Encroach Node=142362.0
       1    3500    5130       0       0       0       0       0       0
       1    3500    5130
Encroach Node=142337.0
       1    3500    5130       0       0       0       0       0       0
       1    3500    5130
Encroach Node=142311.7
       1    3500    5130       0       0       0       0       0       0
       1    3500    5130
Encroach Node=142230.2
       1    3500    5130       0       0       0       0       0       0
       1    3500    5130
Encroach Node=142148.7
       1    3500    5130       0       0       0       0       0       0
       1    3500    5130
Encroach Node=142136.2
       1    3500    5130       0       0       0       0       0       0
       1    3500    5130
Encroach Node=142111.2
       1    3500    5130       0       0       0       0       0       0
       1    3500    5130
Encroach Node=142086.2
       1    3500    5130       0       0       0       0       0       0
       1    3500    5130
Encroach Node=141683.0
       1    3840 5106.94       0       0       0       0       0       0
       1    3840 5106.94
Encroach Node=141165.0
       1    4050    5100       0       0       0       0       0       0
       1    4050    5100
Encroach Node=139993.5
       1    4625    5680       0       0       0       0       0       0
       1    4625    5680
Encroach Node=138970.6
       1    4900 5978.69       0       0       0       0       0       0
       1    4900 5978.69
Encroach Node=138369.4
       1 4862.49    5750       0       0       0       0       0       0
       1 4862.49    5750
Encroach Node=137998.6
       1  4882.9    5500       0       0       0       0       0       0
       1  4882.9    5500
Encroach Node=137941.1
       1  4882.9    5500       0       0       0       0       0       0
       1  4882.9    5500
Encroach Node=137883.6
       1  4882.9    5500       0       0       0       0       0       0
       1  4882.9    5500
Encroach Node=137185.1
       1    4860    5650       0       0       0       0       0       0
       1    4860    5650
Encroach Node=136217.7
       1    4900    5850       0       0       0       0       0       0
       1    4900    5850
Encroach Node=135364.5
       1    4840    5850       0       0       0       0       0       0
       1    4840    5850
Encroach Node=134362.1
       1    4600    5750       0       0       0       0       0       0
       1    4600    5750
Encroach Node=133393.7
       1    4275    5550       0       0       0       0       0       0
       1    4275    5550
Encroach Node=132316.5
       1    4500    5550       0       0       0       0       0       0
       1    4500    5550
Encroach Node=131297.2
       1    4550    5315       0       0       0       0       0       0
       1    4550    5315
Encroach Node=130839.9
       1    4500    5550       0       0       0       0       0       0
       1    4500    5550
Encroach Node=130389.5
       1    4525    5660       0       0       0       0       0       0
       1    4525    6250
Encroach Node=130335.0
       1  4755.8    5670       0       0       0       0       0       0
       1  4755.8    6250
Encroach Node=130280.5
       1  4755.8    5660       0       0       0       0       0       0
       1  4755.8    6250
Encroach Node=130240.5
       1  4755.8    5682       0       0       0       0       0       0
       1  4755.8    6250
Encroach Node=130220.5
       1  4805.2    5672       0       0       0       0       0       0
       1  4805.2    6250
Encroach Node=129735.9
       1  4694.7  5541.5       0       0       0       0       0       0
       1  4694.7    5950
Encroach Node=128777
       1  4669.2    6350       0       0       0       0       0       0
       1  4669.2    6000
Encroach Node=128678.4
       1  4632.2    6500       0       0       0       0       0       0
       1  4632.2    6000
Encroach Node=127716.5
       1  4528.1    6220       0       0       0       0       0       0
       1  4528.1    6200
Encroach Node=126572.3
       1  4555.3    6300       0       0       0       0       0       0
       1  4555.3    6300
Encroach Node=125632.1
       1 4675.56    6000       0       0       0       0       0       0
       1 4675.56    6000
Encroach Node=125012.0
       1 4713.82    5975       0       0       0       0       0       0
       1 4713.82    5975
Encroach Node=124440.5
       1 4683.66    5750       0       0       0       0       0       0
       1 4683.66    5750
Encroach Node=123660.1
       1    4700    5350       0       0       0       0       0       0
       1    4700    5350
Encroach Node=122757.9
       1    4500    5500       0       0       0       0       0       0
       1    4500    5500
Encroach Node=122715.4
       1    4850    5160       0       0       0       0       0       0
       1    4850    5160
Encroach Node=122671.0
       1    4850    5160       0       0       0       0       0       0
       1    4850    5160
Encroach Node=122556.0
       1    4850    5160       0       0       0       0       0       0
       1    4850    5160
Encroach Node=122441.0
       1    4850    5160       0       0       0       0       0       0
       1    4850    5160
Encroach Node=122362.3
       1    4500    5500       0       0       0       0       0       0
       1    4500    5500
Encroach Node=122319.8
       1    4500    5500       0       0       0       0       0       0
       1    4500    5500
Encroach Node=122277.3
       1    4500    5500       0       0       0       0       0       0
       1    4500    5500
Encroach Node=121558.5
       1    4830    5150       0       0       0       0       0       0
       1    4830    5150
Encroach Node=121265.9
       1    4850    5600       0       0       0       0       0       0
       1    4850    5600
Encroach Node=120963.2
       1    4825    7100       0       0       0       0       0       0
       1    4825    7100
Encroach Node=120878.2
       1    4800    7100       0       0       0       0       0       0
       1    4800    7100
Encroach Node=120849.2
       1    4800    7100       0       0       0       0       0       0
       1    4800    7100
Encroach Node=119851.8
       1    4900    7600       0       0       0       0       0       0
       1    4900    7600
Encroach Node=119077.8
       1  4852.6    7600       0       0       0       0       0       0
       1  4852.6    7600
Encroach Node=118735.0
       1  4852.6    7490       0       0       0       0       0       0
       1  4852.6    7490
Encroach Node=118720.5
       1  4852.6    7425       0       0       0       0       0       0
       1  4852.6    7425
Encroach Node=118706.0
       1  4852.6    7385       0       0       0       0       0       0
       1  4852.6    7385
Encroach Node=117895.1
       1    4500    6400       0       0       0       0       0       0
       1    4500    6400
Encroach Node=116691.9
       1    4300    6300       0       0       0       0       0       0
       1    4300    6300
Encroach Node=115756.0
       1    4050    6200       0       0       0       0       0       0
       1    4050    6200
Encroach Node=114790.0
       1    3750    6500       0       0       0       0       0       0
       1    3750    6500
Encroach Node=113752.5
       1    4200    6700       0       0       0       0       0       0
       1    4200    6700
Encroach Node=113002.4
       1    4740    6840       0       0       0       0       0       0
       1    4740    6840
Encroach Node=112280.0
       1    4640    6700       0       0       0       0       0       0
       1    4640    6700
Encroach Node=111431.6
       1    4100    6450       0       0       0       0       0       0
       1    4100    6450
Encroach Node=110232.7
       1    4600    6150       0       0       0       0       0       0
       1    4600    6150
Encroach Node=110012
       1    4531    6049       0       0       0       0       0       0
       1    4531    6049
Encroach Node=109732.
       1 4019.24 5874.24       0       0       0       0       0       0
       1 4019.24 5874.24
Encroach Node=109386.5
       1    4060    5700       0       0       0       0       0       0
       1    4060    5700
Encroach Node=109256
       1    4027    5639       0       0       0       0       0       0
       1    4027    5639
Encroach Node=108653.1
       1    3700    5350       0       0       0       0       0       0
       1    3700    5350
Encroach Node=107478.1
       1    4040    5200       0       0       0       0       0       0
       1    4040    5200
Encroach Node=106679.6
       1    4450    5200       0       0       0       0       0       0
       1    4450    5200
Encroach Node=106389.0
       1    4425    5150       0       0       0       0       0       0
       1    4425    5150
Encroach Node=106217.7
       1    4370    5150       0       0       0       0       0       0
       1    4370    5150
Encroach Node=106185.7
       1    4370    5150       0       0       0       0       0       0
       1    4370    5150
Encroach Node=105689.1
       1    4200    5200       0       0       0       0       0       0
       1    4200    5200
Encroach Node=105015
       1 4132.51 5667.51       0       0       0       0       0       0
       1 4132.51 5667.51
Encroach Node=104955
       1 4119.39 5889.39       0       0       0       0       0       0
       1 4119.39 5889.39
Encroach Node=104781
       1 4119.39 5889.39       0       0       0       0       0       0
       1 4119.39 5889.39
Encroach Node=104697
       1    4100    6000       0       0       0       0       0       0
       1    4100    6000
Encroach Node=104631.0
       1    4100    6000       0       0       0       0       0       0
       1    4100    6000
Encroach Node=103765.5
       1    3770    6590       0       0       0       0       0       0
       1    3770    6590
Encroach Node=103112.4
       1    3500    6985       0       0       0       0       0       0
       1    3500    6985
Encroach Node=102501.5
       1    3900    7300       0       0       0       0       0       0
       1    3900    7300
Encroach Node=101444.8
       1    4030    7400       0       0       0       0       0       0
       1    4030    7400
Encroach Node=100298.8
       1    2800    7460       0       0       0       0       0       0
       1    2800    7460
Encroach Node=99730.8
       1    2400    7230       0       0       0       0       0       0
       1    2400    7230
Encroach Node=99011.4
       1    2200    6720       0       0       0       0       0       0
       1    2200    6720
Encroach Node=98142.3
       1    2400    6080       0       0       0       0       0       0
       1    2400    6080
Encroach Node=97699.3
       1    2600    5900       0       0       0       0       0       0
       1    2600    5900
Encroach Node=97688.8
       1    2600    5900       0       0       0       0       0       0
       1    2600    5900
Encroach Node=97678.3
       1    2600    5900       0       0       0       0       0       0
       1    2600    5900
Encroach Node=97040.1
       1    2750    6200       0       0       0       0       0       0
       1    2750    6200
Encroach Node=95922.1
       1    3600    7050       0       0       0       0       0       0
       1    3600    7050
Encroach Node=95197.2
       1    4000    7340       0       0       0       0       0       0
       1    4000    7340
Encroach Node=94381.9
       1    4500    7800       0       0       0       0       0       0
       1    4500    7800
Encroach Node=93820.0
       1    4400    7600       0       0       0       0       0       0
       1    4400    7600
Encroach Node=92895.0
       1    4400    5760       0       0       0       0       0       0
       1    4400    5760
Encroach Node=91777.0
       1    4240    6080       0       0       0       0       0       0
       1    4240    6080
Encroach Node=90792.7
       1    4899    5091       0       0       0       0       0       0
       1    4899    5091
Encroach Node=90777.7
       1    4899    5091       0       0       0       0       0       0
       1    4899    5091
Encroach Node=90762.7
       1    4899    5091       0       0       0       0       0       0
       1    4899    5091
Encroach Node=90179.9
       1  4885.7    5850       0       0       0       0       0       0
       1  4885.7    5850
Encroach Node=89091.7
       1    4550    5700       0       0       0       0       0       0
       1    4550    5700
Encroach Node=88224.9
       1    4200    5150       0       0       0       0       0       0
       1    4200    5150
Encroach Node=87388.4
       1    4862    5120       0       0       0       0       0       0
       1    4862    5120
Encroach Node=87347.9
       1    4862    5120       0       0       0       0       0       0
       1    4862    5120
Encroach Node=87307.4
       1    4862    5120       0       0       0       0       0       0
       1    4862    5120
Encroach Node=86768.9
       1    4300  5152.7       0       0       0       0       0       0
       1    4300  5152.7
Encroach Node=85988.8
       1    4250    5170       0       0       0       0       0       0
       1    4250    5170
Encroach Node=85105.8
       1    4700    5170       0       0       0       0       0       0
       1    4700    5170
Encroach Node=84426.2
       1    4550    5163       0       0       0       0       0       0
       1    4550    5163
Encroach Node=83474.7
       1    4500    5450       0       0       0       0       0       0
       1    4500    5450
Encroach Node=82559.5
       1    4650    5700       0       0       0       0       0       0
       1    4650    5700
Encroach Node=81700.8
       1  4886.6    6550       0       0       0       0       0       0
       1  4886.6    6550
Encroach Node=80779.8
       1    4830    5700       0       0       0       0       0       0
       1    4830    5700
Encroach Node=80215.8
       1    4780    6090       0       0       0       0       0       0
       1    4780    6090
Encroach Node=79493.4
       1    4760    5100       0       0       0       0       0       0
       1    4760    5100
Encroach Node=78440.2
       1    4850    5110       0       0       0       0       0       0
       1    4850    5110
Encroach Node=77408.6
       1    4850    5150       0       0       0       0       0       0
       1    4850    5150
Encroach Node=76357.2
       1    4800  5100.4       0       0       0       0       0       0
       1    4800  5100.4
Encroach Node=75672.1
       1    4850    5100       0       0       0       0       0       0
       1    4850    5100
Encroach Node=75099.9
       1    4900  5093.6       0       0       0       0       0       0
       1    4900  5093.6
Encroach Node=74185.2
       1    4900    5160       0       0       0       0       0       0
       1    4900    5160
Encroach Node=73452.4
       1    4700    5210       0       0       0       0       0       0
       1    4700    5210
Encroach Node=73270.0
       1    4700    5270       0       0       0       0       0       0
       1    4700    5270
Encroach Node=73221.0
       1    4700    5270       0       0       0       0       0       0
       1    4700    5270
Encroach Node=73172.0
       1    4700    5270       0       0       0       0       0       0
       1    4700    5270
Encroach Node=72763.6
       1    4850    5350       0       0       0       0       0       0
       1    4850    5350
Encroach Node=71993.7
       1    4850    5370       0       0       0       0       0       0
       1    4850    5370
Encroach Node=71075.4
       1    4850    6150       0       0       0       0       0       0
       1    4850    6150
Encroach Node=70236.2
       1    4820    6180       0       0       0       0       0       0
       1    4820    6180
Encroach Node=69380.8
       1    4700    5143       0       0       0       0       0       0
       1    4700    5143
Encroach Node=69172.5
       1    4580    5235       0       0       0       0       0       0
       1    4580    5235
Encroach Node=69141.5
       1    4580    5235       0       0       0       0       0       0
       1    4580    5235
Encroach Node=69110.5
       1    4580    5235       0       0       0       0       0       0
       1    4580    5235
Encroach Node=68465.6
       1    4650    5200       0       0       0       0       0       0
       1    4650    5200
Encroach Node=67438.1
       1    4760    5140       0       0       0       0       0       0
       1    4760    5140
Encroach Node=67045.0
       1    4770    5200       0       0       0       0       0       0
       1    4770    5200
Encroach Node=66490.4
       1    4850    5200       0       0       0       0       0       0
       1    4850    5200
Encroach Node=66476.4
       1    4850    5200       0       0       0       0       0       0
       1    4850    5200
Encroach Node=66462.4
       1    4850    5200       0       0       0       0       0       0
       1    4850    5200
Encroach Node=66068.2
       1    4800    5200       0       0       0       0       0       0
       1    4800    5200
Encroach Node=66051.7
       1    4800    5200       0       0       0       0       0       0
       1    4800    5200
Encroach Node=66035.2
       1    4800    5200       0       0       0       0       0       0
       1    4800    5200
Encroach Node=65928.4
       1    4800    5200       0       0       0       0       0       0
       1    4800    5200
Encroach Node=65087.6
       1    4800    5200       0       0       0       0       0       0
       1    4800    5200
Encroach Node=64048.7
       1    4350    5200       0       0       0       0       0       0
       1    4350    5200
Encroach Node=63532.5
       1    4350    5250       0       0       0       0       0       0
       1    4350    5250
Encroach Node=63354.4
       1    4350    5250       0       0       0       0       0       0
       1    4350    5250
Encroach Node=63339.4
       1    4350    5250       0       0       0       0       0       0
       1    4350    5250
Encroach Node=63324.4
       1    4350    5250       0       0       0       0       0       0
       1    4350    5250
Encroach Node=62095.8
       1    4800    5500       0       0       0       0       0       0
       1    4800    5500
Encroach Node=61100.3
       1    4600    5225       0       0       0       0       0       0
       1    4600    5225
Encroach Node=60007.6
       1    4820    5170       0       0       0       0       0       0
       1    4820    5170
Encroach Node=58881.2
       1    4750    5170       0       0       0       0       0       0
       1    4750    5170
Encroach Node=58492.6
       1    4675    5150       0       0       0       0       0       0
       1    4675    5150
Encroach Node=57991.2
       1    4775    5170       0       0       0       0       0       0
       1    4775    5170
Encroach Node=57964.2
       1    4775    5170       0       0       0       0       0       0
       1    4775    5170
Encroach Node=57937.2
       1    4775    5170       0       0       0       0       0       0
       1    4775    5170
Encroach Node=57897.1
       1    4723    5170       0       0       0       0       0       0
       1    4723    5170
Encroach Node=57861.1
       1    4723    5170       0       0       0       0       0       0
       1    4723    5170
Encroach Node=57825.1
       1    4723    5170       0       0       0       0       0       0
       1    4723    5170
Encroach Node=56911.1
       1    4650    5330       0       0       0       0       0       0
       1    4650    5330
Encroach Node=56116.0
       1    4380    5170       0       0       0       0       0       0
       1    4380    5170
Encroach Node=55154.4
       1    4085    5160       0       0       0       0       0       0
       1    4085    5160
Encroach Node=54063.3
       1    4700    5800       0       0       0       0       0       0
       1    4700    5800
Encroach Node=52958.0
       1    4400    5120       0       0       0       0       0       0
       1    4400    5120
Encroach Node=52205.4
       1    4450    5180       0       0       0       0       0       0
       1    4450    5180
Encroach Node=51121.1
       1    4600    5270       0       0       0       0       0       0
       1    4600    5270
Encroach Node=50135.0
       1    4800    5600       0       0       0       0       0       0
       1    4800    5600
Encroach Node=48853.4
       1    4690    5220       0       0       0       0       0       0
       1    4690    5220
Encroach Node=48177.2
       1    4700    5130       0       0       0       0       0       0
       1    4700    5130
Encroach Node=47168.6
       1    4700    5100       0       0       0       0       0       0
       1    4700    5100
Encroach Node=46018.3
       1    4800    5550       0       0       0       0       0       0
       1    4800    5550
Encroach Node=44828.1
       1    4820    5700       0       0       0       0       0       0
       1    4820    5700
Encroach Node=44797.6
       1    4820    5700       0       0       0       0       0       0
       1    4820    5700
Encroach Node=44767.1
       1    4820    5700       0       0       0       0       0       0
       1    4820    5700
Encroach Node=44499.9
       1    4662    5450       0       0       0       0       0       0
       1    4662    5450
Encroach Node=44470.9
       1    4662    5450       0       0       0       0       0       0
       1    4662    5450
Encroach Node=44441.9
       1    4662    5450       0       0       0       0       0       0
       1    4662    5450
Encroach Node=43183.7
       1    4550    5150       0       0       0       0       0       0
       1    4550    5150
Encroach Node=42427.2
       1    4600    5170       0       0       0       0       0       0
       1    4600    5170
Encroach Node=42387.2
       1    4600    5170       0       0       0       0       0       0
       1    4600    5170
Encroach Node=42347.2
       1    4600    5170       0       0       0       0       0       0
       1    4600    5170
Encroach Node=41330.0
       1    4650    5300       0       0       0       0       0       0
       1    4650    5300
Encroach Node=40345.9
       1    4615    5250       0       0       0       0       0       0
       1    4615    5250
Encroach Node=39549.7
       1    4600    5200       0       0       0       0       0       0
       1    4600    5200
Encroach Node=39013.7
       1    4800    5300       0       0       0       0       0       0
       1    4800    5300
Encroach Node=38132.0
       1    4800    5800       0       0       0       0       0       0
       1    4800    5800
Encroach Node=37339.3
       1  4912.8    6000       0       0       0       0       0       0
       1  4912.8    6000
Encroach Node=36648.9
       1    4800    5300       0       0       0       0       0       0
       1    4800    5300
Encroach Node=36053.8
       1    4800    5300       0       0       0       0       0       0
       1    4800    5300
Encroach Node=35277.3
       1    4780    5175       0       0       0       0       0       0
       1    4780    5175
Encroach Node=35037.7
       1    4500    5220       0       0       0       0       0       0
       1    4500    5220
Encroach Node=34970.2
       1    4500    5220       0       0       0       0       0       0
       1    4500    5220
Encroach Node=34902.7
       1    4500    5220       0       0       0       0       0       0
       1    4500    5220
Encroach Node=34643.9
       1    4770    5520       0       0       0       0       0       0
       1    4770    5520
Encroach Node=34377.0
       1    4740    5600       0       0       0       0       0       0
       1    4740    5600
Encroach Node=33641.9
       1    4900    5220       0       0       0       0       0       0
       1    4900    5220
Encroach Node=32470.2
       1    4820    5260       0       0       0       0       0       0
       1    4820    5260
Encroach Node=31354.3
       1    4790    5150       0       0       0       0       0       0
       1    4790    5150
Encroach Node=30570.5
       1    4472    5130       0       0       0       0       0       0
       1    4472    5130
Encroach Node=29440.5
       1    4800    5260       0       0       0       0       0       0
       1    4800    5260
Encroach Node=28194.0
       1    4450    5140       0       0       0       0       0       0
       1    4450    5140
Encroach Node=27333.4
       1    4570    5230       0       0       0       0       0       0
       1    4570    5230
Encroach Node=26301.3
       1    4680    5120       0       0       0       0       0       0
       1    4680    5120
Encroach Node=25750.5
       1    4460    5180       0       0       0       0       0       0
       1    4460    5180
Encroach Node=25418.2
       1    4360    5480       0       0       0       0       0       0
       1    4360    5480
Encroach Node=25361.7
       1    4360    5480       0       0       0       0       0       0
       1    4360    5480
Encroach Node=25305.2
       1    4360    5480       0       0       0       0       0       0
       1    4360    5480
Encroach Node=24738.4
       1    4500    5500       0       0       0       0       0       0
       1    4500    5500
Encroach Node=24144.0
       1    4600    5360       0       0       0       0       0       0
       1    4600    5360
Encroach Node=23334.1
       1    4675    5200       0       0       0       0       0       0
       1    4675    5200
Encroach Node=22583.9
       1    4725    5470       0       0       0       0       0       0
       1    4725    5470
Encroach Node=21977.3
       1    4800    5450       0       0       0       0       0       0
       1    4800    5450
Encroach Node=21244.2
       1    4900    5500       0       0       0       0       0       0
       1    4900    5500
Encroach Node=20179.5
       1    4800    5330       0       0       0       0       0       0
       1    4800    5330
Encroach Node=19924.3
       1    4741    5242       0       0       0       0       0       0
       1    4741    5242
Encroach Node=19793.3
       1    4741    5242       0       0       0       0       0       0
       1    4741    5242
Encroach Node=19662.3
       1    4741    5242       0       0       0       0       0       0
       1    4741    5242
Encroach Node=18088.1
       1    4300  5134.4       0       0       0       0       0       0
       1    4300  5134.4
Encroach Node=17152.1
       1    4820    5257       0       0       0       0       0       0
       1    4820    5257
Encroach Node=17097.1
       1    4820    5257       0       0       0       0       0       0
       1    4820    5257
Encroach Node=17042.1
       1    4820    5257       0       0       0       0       0       0
       1    4820    5257
Encroach Node=16397.2
       1    4850    5150       0       0       0       0       0       0
       1    4850    5150
Encroach Node=16122.9
       1    4616    5335       0       0       0       0       0       0
       1    4616    5335
Encroach Node=16107.4
       1    4616    5335       0       0       0       0       0       0
       1    4616    5335
Encroach Node=16091.9
       1    4616    5335       0       0       0       0       0       0
       1    4616    5335
Encroach Node=15705.6
       1  4844.7    5300       0       0       0       0       0       0
       1  4844.7    5300
Encroach Node=15477.2
       1  4844.7    5330       0       0       0       0       0       0
       1  4844.7    5330
Encroach Node=15458.7
       1  4844.7    5330       0       0       0       0       0       0
       1  4844.7    5330
Encroach Node=15440.2
       1  4844.7    5330       0       0       0       0       0       0
       1  4844.7    5330
Encroach Node=14412.1
       1    4600  5151.6       0       0       0       0       0       0
       1    4600  5151.6
Encroach Node=13021.2
       1    3650  5139.6       0       0       0       0       0       0
       1    3650  5139.6
Encroach Node=12487.4
       1    3500  5135.4       0       0       0       0       0       0
       1    3500  5135.4
Encroach Node=11271.2
       1    4350  5157.4       0       0       0       0       0       0
       1    4350  5157.4
Encroach Node=10264.8
       1  4855.6  5136.2       0       0       0       0       0       0
       1  4855.6  5136.2
Encroach Node=8988.2
       1  4860.3    5190       0       0       0       0       0       0
       1  4860.3    5190
Encroach Node=7815.2
       1  4849.4  5159.4       0       0       0       0       0       0
       1  4849.4  5159.4
Encroach Node=7068.0
       1  4822.8  5157.3       0       0       0       0       0       0
       1  4822.8  5157.3
Encroach Node=6027.6
       1  4702.9  5233.4       0       0       0       0       0       0
       1  4702.9  5233.4
Encroach Node=5153.0
       1  4770.8  5180.7       0       0       0       0       0       0
       1  4770.8  5180.7
Encroach Node=4272.1
       1  4677.4  5223.3       0       0       0       0       0       0
       1  4677.4  5223.3
Encroach Node=3147.9
       1  4775.7  5207.7       0       0       0       0       0       0
       1  4775.7  5207.7
Encroach Node=2404.5
       1  4769.8  5212.8       0       0       0       0       0       0
       1  4769.8  5212.8
Encroach Node=982.7
       1  4787.2  5212.9       0       0       0       0       0       0
       1  4787.2  5212.9
BEGIN DESCRIPTION:
FEMA Effective Floodway June 2007 + ... + LOMR 13-06-2759P+ LOMR 20-06-2000P
END DESCRIPTION:
Computation Interval=1HOUR
Output Interval=1HOUR
Instantaneous Interval=1HOUR
Mapping Interval=1HOUR
Computation Time Step Use Courant=        0
Computation Time Step Use Time Series=    0
Computation Time Step Count To Double=0
Computation Time Step Max Doubling=0
Computation Time Step Max Halving=0
Computation Time Step Residence Courant=0
Run HTab= 0
Run UNet= 0
Run Sediment= 0
Run PostProcess= 0
Run WQNet= 0
Run RASMapper= 0
UNET Theta= 1
UNET Theta Warmup= 1
UNET ZTol= 0.02
UNET ZSATol= 0.1
UNET MxIter= 20
UNET Max Iter WO Improvement= 0
UNET MaxInSteps= 20
UNET DtIC= 0
UNET DtMin= 0
UNET MaxCRTS= 20
UNET WFStab= 2
UNET SFStab= 1
UNET WFX= 1
UNET SFX= 1
UNET 1D Methodology=Finite Difference
UNET DSS MLevel= 4
UNET Pardiso=0
UNET DZMax Abort= 100
UNET Use Existing IB Tables=-1
UNET Froude Reduction=False
UNET Froude Limit= 0.8
UNET Froude Power= 4
UNET D1 Cores= 0
UNET D2 Coriolis=0
UNET D2 Cores= 0
UNET D2 Theta= 1
UNET D2 Theta Warmup= 1
UNET D2 Z Tol= 0.01
UNET D2 Volume Tol= 0.01
UNET D2 Max Iterations= 20
UNET D2 Equation= 0
UNET D2 RampUpFraction=0.1
UNET D2 TimeSlices= 1
UNET D2 BCVolumeCheck=0
UNET D1D2 MaxIter= 0
UNET D1D2 ZTol=0.01
UNET D1D2 QTol=0.1
UNET D1D2 MinQTol=1
Write IC File= 0
Write IC File at Fixed DateTime=0
IC Time=0,,
Write IC File at Sim End=0
Echo Input=False
Echo Parameters=False
Echo Output=False
Write Detailed= 0
HDF Write Warmup=0
HDF Write Time Slices=0
HDF Flush=0
HDF Face Node Velocities=0
HDF Compression= 1
HDF Chunk Size= 1
HDF Spatial Parts= 1
HDF Use Max Rows=0
HDF Fixed Rows= 1
Calibration Method= 0
Calibration Iterations= 20
Calibration Max Change=0.05
Calibration Tolerance=0.2
Calibration Maximum=1.5
Calibration Minimum=0.5
Calibration Optimization Method= 1
WQ AD Non Conservative
WQ ULTIMATE=-1
WQ Max Comp Step=1HOUR
WQ Output Interval=15MIN
WQ Output Selected Increments= 0
WQ Output face flow=0
WQ Output face velocity=0
WQ Output face area=0
WQ Output face dispersion=0
WQ Output cell volume=0
WQ Output cell surface area=0
WQ Output cell continuity=0
WQ Output cumulative cell continuity=0
WQ Output face conc=0
WQ Output face dconc_dx=0
WQ Output face courant=0
WQ Output face peclet=0
WQ Output face adv mass=0
WQ Output face disp mass=0
WQ Output cell mass=0
WQ Output cell source sink temp=0
WQ Output nsm pathways=0
WQ Output nsm derived pathways=0
WQ Output MaxMinRange=-1
WQ Daily Max Min Mean=-1
WQ Daily Range=0
WQ Daily Time=0
WQ Create Restart=0
WQ Fixed Restart=0
WQ System Summary=0
WQ Write To DSS=0
WQ Use Fixed Temperature=0
Sorting and Armoring Iterations= 10
XS Update Threshold= 0.02
Bed Roughness Predictor= 0
Hydraulics Update Threshold= 0.02
Energy Slope Method= 1
Volume Change Method= 1
Sediment Retention Method= 0
XS Weighting Method= 0
Number of US Weighted Cross Sections= 1
Number of DS Weighted Cross Sections= 1
Upstream XS Weight=0
Main XS Weight=1
Downstream XS Weight=0
Number of DS XS's Weighted with US Boundary= 1
Upstream Boundary Weight= 1
Weight of XSs Associated with US Boundary= 0
Number of US XS's Weighted with DS Boundary= 1
Downstream Boundary Weight= 0.5
Weight of XSs Associated with DS Boundary= 0.5
Percentile Method= 0
Sediment Output Level= 3
Mass or Volume Output= 0
Output Increment Type= 1
Profile and TS Output Increment= 1
XS Output Flag= 0
XS Output Increment= 10
Write Gradation File= 0
Read Gradation Hotstart= 0
Write HDF5 File= 1
Write Binary Output= 1
Write DSS Sediment File= 0
SV Curve= 0
Specific Gage Flag= 0
