HEC-RAS study P100-00-00.prj: P100-00-00

--- P100-00-00.g01 (geometry) --- (continued)

Type RM Length L Ch R = 3 ,210776.9,,,
BEGIN DESCRIPTION:
FM 249 TOMBALL PARKWAY - 45 degree skew
Structure ID: P00-84
END DESCRIPTION:
Bridge Culvert--1,0,-1,-1, 0
Deck Dist Width WeirC Skew NumUp NumDn MinLoCord MaxHiCord MaxSubmerge Is_Ogee
10,560,2.6,0, 60, 60, , , 0.95, 0, 1,1,,
  2735.5  2814.7  2879.3  2999.3  3049.3    3457    3507    3687    3717    3784
    3824    3884    4034  4246.4  4507.8  4697.8  4744.5 4779.78 4793.71 4874.59
  4874.7 4888.49 4912.27 4912.36 5079.73  5151.6 5188.86 5189.14 5314.02  5352.7
  5402.7  5581.2 5581.31  5582.7  5628.8  6222.7  6322.7  6412.7  6502.7  6532.7
  6572.7  6602.7  6802.7  6822.7  6842.7  7002.7  7082.7  7112.7  7162.7  7202.7
  7262.7  7492.7  7522.7  7542.7  7562.7  7572.7  7592.7  7652.7    7783  7788.7
   120.7   127.5  127.48  127.44  127.42  127.28  127.26   127.2  127.18  127.16
  127.15  127.13  127.07     127  123.74  121.38  120.75  120.17  119.97     119
   120.6  120.57  120.51  120.51  120.68  120.78  120.75  120.75  120.38  120.35
   120.4  120.45  118.85  118.85  118.86  118.92  118.93  118.94  118.95  118.95
  118.96  118.96  118.98  118.98  118.99  118.99  118.94  118.92  118.89  118.86
  118.82  118.68  118.66  118.65  118.64  118.63  118.62  118.58   118.5   118.6
   120.7   120.9   119.1   118.2   119.3   118.8   117.5   116.1   114.5   115.6
     115   116.4   115.9   116.6   116.8   118.2  117.31   118.9  118.07  117.37
  117.37  117.25  115.56  116.61  116.39  117.51  116.17  115.63  117.01   115.2
   116.4  114.12  114.12   114.1     115   117.6   116.2   115.9   116.1   117.3
   116.1   117.8   117.6     116   112.9   112.3   113.5     115   115.2   114.5
   116.4   115.3   116.5   115.8   113.6   113.3   115.3   116.3   116.2   118.6
  2735.5  2814.7  2879.3  2999.3  3049.3    3457    3507    3687    3717    3784
    3824    3884    4034  4246.4  4507.8  4697.8  4744.5 4779.78 4793.71 4874.59
  4874.7 4888.49 4912.27 4912.36 5079.73  5151.6 5188.86 5189.14 5314.02  5352.7
  5402.7  5581.2 5581.31  5582.7  5628.8  6222.7  6322.7  6412.7  6502.7  6532.7
  6572.7  6602.7  6802.7  6822.7  6842.7  7002.7  7082.7  7112.7  7162.7  7202.7
  7262.7  7492.7  7522.7  7542.7  7562.7  7572.7  7592.7  7652.7    7783  7788.7
   120.7   127.5  127.48  127.44  127.42  127.28  127.26   127.2  127.18  127.16
  127.15  127.13  127.07     127  123.74  121.38  120.75  120.17  119.97     119
   120.6  120.57  120.51  120.51  120.68  120.78  120.75  120.75  120.38  120.35
   120.4  120.45  118.85  118.85  118.86  118.92  118.93  118.94  118.95  118.95
  118.96  118.96  118.98  118.98  118.99  118.99  118.94  118.92  118.89  118.86
  118.82  118.68  118.66  118.65  118.64  118.63  118.62  118.58   118.5   118.6
  120.62  120.82  119.02  118.12  119.22  118.72  117.42  116.02  114.42  115.52
  114.92  116.32  115.82  116.52  116.72  118.12  117.23  118.82  117.99  117.29
  117.29  117.17  115.48  116.53  116.31  117.43  116.09  115.55  116.93  115.12
  116.32  114.04  114.04  114.02  114.92  117.52  116.12  115.82  116.02  117.22
  116.02  117.72  117.52  115.92  112.82  112.22  113.42  114.92  115.12  114.42
  116.32  115.22  116.42  115.72  113.52  113.22  115.22  116.22  116.12  118.52
Pier Skew, UpSta & Num, DnSta & Num=  ,4954.6, 2 ,4954.6, 2 , 0 , 0 , 0 ,,
     1.4     1.4
  105.62  117.53
     1.4     1.4
  105.54  117.45
Pier Skew, UpSta & Num, DnSta & Num=  ,4996.4, 2 ,4996.4, 2 , 0 , 0 , 0 ,,
     1.4     1.4
  102.53  117.46
     1.4     1.4
  102.45  117.38
Pier Skew, UpSta & Num, DnSta & Num=  ,5038, 2 ,5038, 2 , 0 , 0 , 0 ,,
     1.4     1.4
  103.94   117.6
     1.4     1.4
  103.86  117.52
Abutment Skew #Up #Dn= , 2 , 2
 4912.16 4937.77
  116.61  106.28
 4912.16 4937.77
  116.53   106.2
Abutment Skew #Up #Dn= , 2 , 2
 5053.69 5079.82
  105.51  116.78
 5053.69 5079.82
  105.43   116.7
BR Coef= 1 , 1 , 0 ,1.25, 0 ,,,0.8,0,2,0,
WSPro=,,,, 1 ,,,, 0 ,,,, 0 ,,,,-1 ,-1 ,-1 , 0 , 0 , 0 , 0 , 0
BR U #Sta/Elev= 122
  2735.5   120.7  2814.7   120.9  2815.5   120.9  2819.3   120.8  2879.3   119.1
  2999.3   118.2  3049.3   119.3    3147   118.9    3237   118.6    3457   118.8
    3507   117.5    3687   116.1    3717   114.5    3724   114.5    3784   115.6
    3824     115    3884   116.4    4034   115.9    4054   116.3  4246.4   116.6
    4374   116.8    4394   116.4  4507.8   116.8  4697.8   118.2  4730.6  117.57
  4730.9  117.57  4744.5  117.31 4779.78   118.9  4789.7  118.31 4793.71  118.07
  4856.5  117.53 4874.59  117.37  4874.7  117.37 4874.81  117.37 4888.49  117.25
 4912.27  115.56 4912.36  115.56 4917.54  115.19  4929.7  109.81 4937.57  106.32
 4937.67  106.28 4952.68  106.31 4954.64  106.79 4969.41  104.96  4985.7  104.98
 4991.46  104.99 4996.36  103.48 4999.16  103.68 5001.47  102.45 5003.36   103.1
  5004.5  103.76 5008.54   106.1 5011.62   105.4 5024.85  104.58 5026.53  103.55
 5038.01  105.03 5053.59  105.39 5053.69  105.51 5062.65  115.87 5079.62  116.38
 5079.73  116.39    5086  116.58 5088.13  116.64 5101.15  116.71  5113.9  116.91
  5151.6  117.51  5158.2  117.62 5188.86  116.17 5189.14  115.63 5211.19   115.7
 5213.43  116.08  5240.2  116.33 5314.02  117.01  5325.5  116.57  5332.7   116.3
  5352.7   115.2  5402.7   116.4  5425.4  116.11  5508.7  115.05    5581  114.12
 5581.09  114.12  5581.2  114.12 5581.31  114.12  5582.7   114.1  5628.8     115
  5988.8   116.7  5998.8   116.4  6122.7   116.8  6222.7   117.6  6322.7   116.2
  6412.7   115.9  6502.7   116.1  6532.7   117.3  6552.7     117  6572.7   116.1
  6602.7   117.8  6752.7   117.4  6802.7   117.6  6822.7     116  6832.7     114
  6842.7   112.9  6979.2  112.39  7002.7   112.3  7082.7   113.5  7112.7     115
  7162.7   115.2  7172.7   114.8  7182.7     115  7202.7   114.5  7232.7   115.3
  7262.7   116.4  7492.7   115.3  7522.7   116.5  7542.7   115.8  7552.7   114.5
  7562.7   113.6  7572.7   113.3  7592.7   115.3  7652.7   116.3    7783   116.2
  7787.6  118.14  7788.7   118.6
BR U #Mann= 3
  2735.5      .1 4917.54    .035 5088.13      .1
BR U Banks=4917.54,5088.13
BR D #Sta/Elev= 122
  2735.5  120.62  2814.7  120.82  2815.5  120.82  2819.3  120.72  2879.3  119.02
  2999.3  118.12  3049.3  119.22    3147  118.82    3237  118.52    3457  118.72
    3507  117.42    3687  116.02    3717  114.42    3724  114.42    3784  115.52
    3824  114.92    3884  116.32    4034  115.82    4054  116.22  4246.4  116.52
    4374  116.72    4394  116.32  4507.8  116.72  4697.8  118.12  4730.6  117.49
  4730.9  117.49  4744.5  117.23 4779.78  118.82  4789.7  118.23 4793.71  117.99
  4856.5  117.45 4874.59  117.29  4874.7  117.29 4874.81  117.29 4888.49  117.17
 4912.27  115.48 4912.36  115.48 4917.54  115.11  4929.7  109.73 4937.57  106.24
 4937.67   106.2 4952.68  106.23 4954.64  106.71 4969.41  104.88  4985.7   104.9
 4991.46  104.91 4996.36   103.4 4999.16   103.6 5001.47  102.37 5003.36  103.02
  5004.5  103.68 5008.54  106.02 5011.62  105.32 5024.85   104.5 5026.53  103.47
 5038.01  104.95 5053.59  105.31 5053.69  105.43 5062.65  115.79 5079.62   116.3
 5079.73  116.31    5086   116.5 5088.13  116.56 5101.15  116.63  5113.9  116.83
  5151.6  117.43  5158.2  117.54 5188.86  116.09 5189.14  115.55 5211.19  115.62
 5213.43     116  5240.2  116.25 5314.02  116.93  5325.5  116.49  5332.7  116.22
  5352.7  115.12  5402.7  116.32  5425.4  116.03  5508.7  114.97    5581  114.04
 5581.09  114.04  5581.2  114.04 5581.31  114.04  5582.7  114.02  5628.8  114.92
  5988.8  116.62  5998.8  116.32  6122.7  116.72  6222.7  117.52  6322.7  116.12
  6412.7  115.82  6502.7  116.02  6532.7  117.22  6552.7  116.92  6572.7  116.02
  6602.7  117.72  6752.7  117.32  6802.7  117.52  6822.7  115.92  6832.7  113.92
  6842.7  112.82  6979.2  112.31  7002.7  112.22  7082.7  113.42  7112.7  114.92
  7162.7  115.12  7172.7  114.72  7182.7  114.92  7202.7  114.42  7232.7  115.22
  7262.7  116.32  7492.7  115.22  7522.7  116.42  7542.7  115.72  7552.7  114.42
  7562.7  113.52  7572.7  113.22  7592.7  115.22  7652.7  116.22    7783  116.12
  7787.6  118.06  7788.7  118.52
BR D #Mann= 3
  2735.5      .1 4917.54    .035 5088.13      .1
BR D Banks=4917.54,5088.13
BC Design=,, 0 ,, 0 ,,,,,,
BC HTab HWMax=120.9
BC Use User HTab Curves=0
BC User HTab FreeFlow(D)= 0

Type RM Length L Ch R = 1 ,210486.9,464.2,464.2,464.2
BEGIN DESCRIPTION:
Downstream Section of Bridge/Culvert/Weir
END DESCRIPTION:
XS GIS Cut Line= 6
      3064456.31     13910879.66      3064730.89     13910660.51
      3066215.25     13909573.25      3066986.58     13908950.28
      3067419.63     13908253.58      3067731.32     13907251.72
#Sta/Elev= 30
  2735.5  120.59  2999.3  118.09    3457  118.69    3717  114.39    3884  116.29
  4744.5   117.2 4779.78  118.79 4917.54  115.08 4937.67  106.17 4991.46  104.88
 5001.47  102.34 5008.54  105.99 5026.53  103.44 5053.59  105.28 5062.65  115.76
 5088.13  116.53 5314.02   116.9  5352.7  115.09  5582.7  113.99  6222.7  117.49
  6412.7  115.79  6802.7  117.49  6842.7  112.79  7002.7  112.19  7262.7  116.29
  7522.7  116.39  7572.7  113.19  7652.7  116.19    7783  116.09  7788.7  118.49
#Mann= 3 , 1 , 0
  2735.5      .1       0 4917.54    .035       0 5088.13      .1       0
#XS Ineff= 2 , 0
       0    4903   119.7    5089       0   118.6
Permanent Ineff=
       F       F
Bank Sta=4917.54,5088.13
XS Rating Curve= 0 ,0
Exp/Cntr=0.5,0.3

Type RM Length L Ch R = 1 ,210022.7,628.9,611.7,483.3
BEGIN DESCRIPTION:
Cross Section 210022.7-Interpolated
END DESCRIPTION:
XS GIS Cut Line= 6
      3064627.26     13911979.11      3066639.07     13909915.68
      3066755.21     13909209.16      3067394.89     13908657.01
        3067500.     13908344.02      3068062.32     13907624.25
#Sta/Elev= 30
  1641.3     122  1926.2   121.5  2176.2   115.5  2326.2   117.2  2446.2   114.6
  3046.2   115.1    3131  116.42  3186.2   115.2  3916.2   115.5  3956.2   118.7
  4006.2     116  4036.2   110.9  4056.2   111.6  4096.2     117  4326.2   115.8
  4476.2   116.9  4569.5   114.3  4829.5   118.2  4947.6  111.37  4981.8  102.06
  5016.4     101  5033.8  109.09  5053.1  112.66  5059.5   114.7  6649.9   117.5
  6755.2  115.89  6989.9   115.3  7139.9     117  7209.9   115.6  7344.1   118.5
#Mann= 5 , 1 , 0
  1641.3      .1       0    3131     .14       0  4947.6    .035       0
  5053.1     .14       0  6755.2      .1       0
#XS Ineff= 2 , 0
       0  4100.2   118.7  6649.9       0   117.5
Permanent Ineff=
       F       F
Bank Sta=4947.6,5053.1
XS Rating Curve= 0 ,0
Exp/Cntr=0.5,0.3

Type RM Length L Ch R = 1 ,209411.0,40,40,40
BEGIN DESCRIPTION:
Upstream Section of Bridge/Culvert/Weir
END DESCRIPTION:
XS GIS Cut Line= 6
      3064378.32      13915062.6       3066774.7     13910535.23
      3066812.32     13910469.72      3067597.25     13909003.61
      3067932.88     13908355.97      3068296.11     13907679.95
#Sta/Elev= 30
 -1278.9  118.96  -685.1  119.41   214.9  115.71  1337.6   116.6  1834.9  117.61
  2054.9  116.01  2614.9  118.91  2954.9  115.31  3144.9  118.21  3424.6  115.71
  3474.6  118.01  3514.6  115.21  3684.6  118.11  3834.6  114.11  4827.3   114.5
  4914.8  114.07  4941.7  110.15  4947.6  111.48  4981.8  102.17  4998.6  100.34
  5016.4  101.11  5033.8   109.2  5053.1  112.77  6161.8  117.71  6231.8  115.81
  6421.8  117.01    6905  115.01  7010.8  118.39  7030.6  118.48    7079  118.71
#Mann= 6 , 1 , 0
 -1278.9      .2       0  1337.6     .14       0  4947.6    .035       0
  5053.1     .14       0  7010.8      .1       0  7030.6      .2       0
#XS Ineff= 2 , 0
       0    4903   118.9    5063       0     119
Permanent Ineff=
       F       F
Bank Sta=4947.6,5053.1
XS Rating Curve= 0 ,0
Exp/Cntr=0.5,0.3

Type RM Length L Ch R = 3 ,209391.0,,,
BEGIN DESCRIPTION:
NORTHERN CENTER RAILROAD
Structure ID: P00-82
END DESCRIPTION:
Bridge Culvert--1,0,-1,-1, 0
Deck Dist Width WeirC Skew NumUp NumDn MinLoCord MaxHiCord MaxSubmerge Is_Ogee
10,20,2.6,0, 60, 60, , , 0.95, 0, 1,1,,
 -1278.9  -685.1  -575.1   214.9   384.9  1594.9  1754.9  1784.9  1804.9  1834.9
  2054.9  2164.9  2194.9  2234.9  2304.9  2344.9  2404.9  2484.9  2524.9  2614.9
  2694.9  2734.9  2854.9  2884.9  2954.9  3094.9  3124.9  3144.9  3384.6  3424.6
  3474.6  3514.6  3684.6  3724.6  3764.6  3804.6  3834.6  4827.3 4914.01  4914.1
    5019 5053.39  5053.5  5055.9  5209.8  5264.5  5399.9  6091.8  6161.8  6231.8
  6311.8  6391.8  6421.8  6531.8    6815    6905    6995  7021.1  7030.6    7079
  118.95  119.41  118.95  118.95  118.94  118.94  118.94  118.94  118.94  118.94
  118.94  118.94  118.94  118.94  118.94  118.94  118.94  118.94  118.94  118.94
  118.94  118.94  118.94  118.94  118.94  118.94  118.94  118.94  118.93  118.93
  118.93  118.93  118.93  118.93  118.93  118.93  118.93  119.04  119.25  119.25
  119.29  119.25  119.25  119.22  119.04  119.07  119.09  119.18  119.19   119.2
  119.21  119.22  119.22  119.24  119.27  119.28   119.3   119.3  118.47   118.7
  118.95   119.4   118.9   115.7   116.9   116.5   117.6   116.1   116.1   117.6
     116     117   116.4   117.3   117.4   118.3   117.6   118.2   117.7   118.9
   117.1   118.2     117   115.7   115.3   117.4   117.4   118.2   116.8   115.7
     118   115.2   118.1   117.7   115.4   115.1   114.1  114.49  114.07  114.75
  114.79  114.75  112.83  113.24  113.61  114.53   115.2     116   117.7   115.8
     117   116.6     117   115.7   115.8     115   118.3  118.42  118.47   118.7
 -1278.9  -685.1  -575.1   214.9   384.9  1594.9  1754.9  1784.9  1804.9  1834.9
  2054.9  2164.9  2194.9  2234.9  2304.9  2344.9  2404.9  2484.9  2524.9  2614.9
  2694.9  2734.9  2854.9  2884.9  2954.9  3094.9  3124.9  3144.9  3384.6  3424.6
  3474.6  3514.6  3684.6  3724.6  3764.6  3804.6  3834.6  4827.3 4914.01  4914.1
    5019 5053.39  5053.5  5055.9  5209.8  5264.5  5399.9  6091.8  6161.8  6231.8
  6311.8  6391.8  6421.8  6531.8    6815    6905    6995  7021.1  7030.6    7079
  118.95  119.41  118.95  118.95  118.94  118.94  118.94  118.94  118.94  118.94
  118.94  118.94  118.94  118.94  118.94  118.94  118.94  118.94  118.94  118.94
  118.94  118.94  118.94  118.94  118.94  118.94  118.94  118.94  118.93  118.93
  118.93  118.93  118.93  118.93  118.93  118.93  118.93  119.04  119.25  119.25
  119.29  119.25  119.25  119.22  119.04  119.07  119.09  119.18  119.19   119.2
  119.21  119.22  119.22  119.24  119.27  119.28   119.3   119.3  118.47   118.7
  118.87  119.32  118.82  115.62  116.82  116.42  117.52  116.02  116.02  117.52
  115.92  116.92  116.32  117.22  117.32  118.22  117.52  118.12  117.62  118.82
  117.02  118.12  116.92  115.62  115.22  117.32  117.32  118.12  116.72  115.62
  117.92  115.12  118.02  117.62  115.32  115.02  114.02  114.41  113.99  114.67
  114.71  114.67  112.75  113.16  113.53  114.45  115.12  115.92  117.62  115.72
  116.92  116.52  116.92  115.62  115.72  114.92  118.22  118.34  118.39  118.62
Pier Skew, UpSta & Num, DnSta & Num=  ,4941.7, 2 ,4941.7, 2 , 0 , 0 , 0 ,,
     1.4     1.4
  109.24  115.78
     1.4     1.4
  109.16   115.7
Pier Skew, UpSta & Num, DnSta & Num=  ,4969.9, 2 ,4969.9, 2 , 0 , 0 , 0 ,,
     1.4     1.4
  104.64   115.8
     1.4     1.4
  104.56  115.72
Pier Skew, UpSta & Num, DnSta & Num=  ,4998.6, 2 ,4998.6, 2 , 0 , 0 , 0 ,,
     1.4     1.4
   99.41  115.81
     1.4     1.4
   99.33  115.73
Pier Skew, UpSta & Num, DnSta & Num=  ,5025.8, 2 ,5025.8, 2 , 0 , 0 , 0 ,,
     1.4     1.4
  105.27  115.78
     1.4     1.4
  105.19   115.7
BR Coef= 1 , 1 , 0 ,1.25, 0 ,,,0.8,0,2,0,
WSPro=,,,, 1 ,,,, 0 ,,,, 0 ,,,,-1 ,-1 ,-1 , 0 , 0 , 0 , 0 , 0
BR U #Sta/Elev= 109
 -1278.9  118.95  -685.1   119.4  -575.1   118.9   214.9   115.7   384.9   116.9
  1337.6  116.59  1594.9   116.5  1754.9   117.6  1784.9   116.1  1804.9   116.1
  1834.9   117.6  2054.9     116  2164.9     117  2194.9   116.4  2234.9   117.3
  2304.9   117.4  2344.9   118.3  2404.9   117.6  2484.9   118.2  2524.9   117.7
  2574.9   118.1  2584.9   118.6  2614.9   118.9  2694.9   117.1  2704.9   117.2
  2734.9   118.2  2854.9     117  2884.9   115.7  2954.9   115.3  3094.9   117.4
  3124.9   117.4  3144.9   118.2  3214.6   118.1  3384.6   116.8  3424.6   115.7
  3434.6   115.8  3464.6   117.8  3474.6     118  3514.6   115.2  3684.6   118.1
  3724.6   117.7  3764.6   115.4  3804.6   115.1  3814.6   114.6  3834.6   114.1
  4666.9  114.27  4678.4   114.3  4722.4  114.29  4781.8  114.28  4784.5  114.28
    4795  114.22    4827  114.49  4827.3  114.49  4850.7  114.24  4902.7  114.22
  4913.4  114.08  4913.9  114.07 4914.01  114.07  4914.1  114.07  4914.2  114.07
  4914.8  114.06  4941.7  110.14  4947.6  111.47  4969.9  105.83    4981  102.78
  4981.8  102.16  4987.2  101.57  4998.6  100.33    5002  101.35  5016.4   101.1
    5019  103.05  5025.8  106.64  5033.8  109.19  5053.1  112.76  5053.3  112.79
 5053.39  112.81  5053.5  112.83  5053.6  112.85  5054.6  113.02  5055.9  113.24
  5151.4  113.73  5152.7  113.74  5209.7  113.61  5209.8  113.61  5264.5  114.53
  5265.3  114.53  5399.9   115.2  5811.8   115.9  5891.8   115.9  6081.8   116.3
  6091.8     116  6111.8   116.7  6151.8   117.2  6161.8   117.7  6181.8   117.5
  6231.8   115.8  6311.8     117  6391.8   116.6  6421.8     117  6531.8   115.7
  6651.8   115.8    6815   115.8    6905     115    6935   115.9    6995   118.3
  7010.8  118.38  7021.1  118.42  7030.6  118.47    7079   118.7
BR U #Mann= 6
 -1278.9      .2  1337.6     .14  4947.6    .035  5053.1     .14  7010.8      .1
  7030.6      .2
BR U Banks=4947.6,5053.1
BR D #Sta/Elev= 109
 -1278.9  118.87  -685.1  119.32  -575.1  118.82   214.9  115.62   384.9  116.82
  1337.6  116.51  1594.9  116.42  1754.9  117.52  1784.9  116.02  1804.9  116.02
  1834.9  117.52  2054.9  115.92  2164.9  116.92  2194.9  116.32  2234.9  117.22
  2304.9  117.32  2344.9  118.22  2404.9  117.52  2484.9  118.12  2524.9  117.62
  2574.9  118.02  2584.9  118.52  2614.9  118.82  2694.9  117.02  2704.9  117.12
  2734.9  118.12  2854.9  116.92  2884.9  115.62  2954.9  115.22  3094.9  117.32
  3124.9  117.32  3144.9  118.12  3214.6  118.02  3384.6  116.72  3424.6  115.62
  3434.6  115.72  3464.6  117.72  3474.6  117.92  3514.6  115.12  3684.6  118.02
  3724.6  117.62  3764.6  115.32  3804.6  115.02  3814.6  114.52  3834.6  114.02
  4666.9  114.19  4678.4  114.22  4722.4  114.21  4781.8   114.2  4784.5   114.2
    4795  114.14    4827  114.41  4827.3  114.41  4850.7  114.16  4902.7  114.14
  4913.4     114  4913.9  113.99 4914.01  113.99  4914.1  113.99  4914.2  113.99
  4914.8  113.98  4941.7  110.06  4947.6  111.39  4969.9  105.75    4981   102.7
  4981.8  102.08  4987.2  101.49  4998.6  100.25    5002  101.27  5016.4  101.02
    5019  102.97  5025.8  106.56  5033.8  109.11  5053.1  112.68  5053.3  112.71
 5053.39  112.73  5053.5  112.75  5053.6  112.77  5054.6  112.94  5055.9  113.16
  5151.4  113.65  5152.7  113.66  5209.7  113.53  5209.8  113.53  5264.5  114.45
  5265.3  114.45  5399.9  115.12  5811.8  115.82  5891.8  115.82  6081.8  116.22
  6091.8  115.92  6111.8  116.62  6151.8  117.12  6161.8  117.62  6181.8  117.42
  6231.8  115.72  6311.8  116.92  6391.8  116.52  6421.8  116.92  6531.8  115.62
  6651.8  115.72    6815  115.72    6905  114.92    6935  115.82    6995  118.22
  7010.8   118.3  7021.1  118.34  7030.6  118.39    7079  118.62
BR D #Mann= 6
 -1278.9      .2  1337.6     .14  4947.6    .035  5053.1     .14  7010.8      .1
  7030.6      .2
BR D Banks=4947.6,5053.1
BC Design=,, 0 ,, 0 ,,,,,,
BC HTab HWMax=119.41
BC Use User HTab Curves=0
BC User HTab FreeFlow(D)= 0

Type RM Length L Ch R = 1 ,209371.0,89.6,89.6,89.6
BEGIN DESCRIPTION:
Downstream Section of Bridge/Culvert/Weir
END DESCRIPTION:
XS GIS Cut Line= 6
      3064418.22     13915065.43       3066814.6     13910538.05
      3066852.22     13910472.54      3067637.15     13909006.43
      3067972.78     13908358.79      3068336.01     13907682.78
#Sta/Elev= 30
 -1278.9  118.88  -685.1  119.33   214.9  115.63  1337.6  116.52  1834.9  117.53
  2054.9  115.93  2614.9  118.83  2954.9  115.23  3144.9  118.13  3424.6  115.63
  3474.6  117.93  3514.6  115.13  3684.6  118.03  3834.6  114.03  4827.3  114.42
  4914.8  113.99  4941.7  110.07  4947.6   111.4  4981.8  102.09  4998.6  100.26
  5016.4  101.03  5033.8  109.12  5053.1  112.69  6161.8  117.63  6231.8  115.73
  6421.8  116.93    6905  114.93  7010.8  118.31  7030.6   118.4    7079  118.63
#Mann= 6 , 1 , 0
 -1278.9      .2       0  1337.6     .14       0  4947.6    .035       0
  5053.1     .14       0  7010.8      .1       0  7030.6      .2       0
#XS Ineff= 2 , 0
       0    4903   118.9    5063       0   118.8
Permanent Ineff=
       F       F
Bank Sta=4947.6,5053.1
XS Rating Curve= 0 ,0
Exp/Cntr=0.5,0.3

Type RM Length L Ch R = 1 ,209281.4,50,50,50
BEGIN DESCRIPTION:
Upstream Section of Bridge/Culvert/Weir
END DESCRIPTION:
XS GIS Cut Line= 6
      3064781.19     13914766.14      3064899.57     13914513.66
      3067394.23     13909647.74      3067459.89     13909513.79
      3067602.44     13909210.87      3068419.67     13907602.65
#Sta/Elev= 30
  -882.6  122.29  -742.6  121.39  -672.6  118.19   761.4  116.69   881.4  117.99
  1061.4  115.29  1379.2  115.62  4804.3  114.24  4943.1  112.87  4948.2  110.26
  4971.7  105.85  4977.5  103.21  4988.9  102.91  4990.3   101.1  4999.3  100.37
  5004.6  102.92  5006.8  101.61  5018.2  103.81  5040.1  114.37  5994.1  116.39
  6054.1  114.99  6074.1  116.79  6114.1  115.29  6174.1  118.29  6214.1  116.99
  6264.1  113.29  6304.1  115.79  6892.3  113.89  7042.3  114.69  7152.3  119.09
#Mann= 4 , 1 , 0
  -882.6      .2       0  1379.2     .14       0  4948.2    .035       0
  5040.1     .14       0
#XS Ineff= 2 , 0
       0    4837   118.5    5130       0   118.5
Permanent Ineff=
       F       F
Bank Sta=4948.2,5040.1
XS Rating Curve= 0 ,0
Exp/Cntr=0.5,0.3

Type RM Length L Ch R = 3 ,209256.4,,,
BEGIN DESCRIPTION:
H. L. & P. ACCESS BRIDGE
Structure ID: P00-81
END DESCRIPTION:
Bridge Culvert--1,0,-1,-1, 0
Deck Dist Width WeirC Skew NumUp NumDn MinLoCord MaxHiCord MaxSubmerge Is_Ogee
10,30,2.6,0, 60, 60, , , 0.95, 0, 1,1,,
  -882.6  -752.6  -742.6  -732.6  -722.6  -672.6  -588.6   -98.6   261.4   761.4
   811.4   851.4   881.4   901.4  1001.4  1061.4  2641.4  2661.4  4094.1  4722.2
  4804.3  4804.7  4881.1  4924.6  4928.9  4943.1  4948.2 4952.31  4952.4 5030.49
  5030.6  5040.1  5068.4  5111.2  5279.4  5574.1  5894.1  5994.1  6054.1  6074.1
  6084.1  6094.1  6114.1  6134.1  6174.1  6194.1  6214.1  6254.1  6264.1  6304.1
  6494.1  6502.3  6612.3  6652.3  6732.3  6852.3  6892.3  7042.3  7092.3  7152.3
   122.3   121.1   121.4   120.9   119.8   118.2   118.5   117.1   117.4   116.7
   117.9   117.3     118   117.2   115.6   115.3   115.9   115.5   114.6   113.6
  114.26  114.07   114.1  113.23  114.15  114.18  114.19   114.2   114.2  114.24
  114.24  114.39  114.66  114.14  114.13   115.6   115.3   116.4     115   116.8
   116.7   115.7   115.3   116.6   118.3   117.2     117   113.6   113.3   115.8
     115   115.3   115.4   114.4     115   114.5   113.9   114.7   117.2   119.1
   122.3   121.1   121.4   120.9   119.8   118.2   118.5   117.1   117.4   116.7
   117.9   117.3     118   117.2   115.6   115.3   115.9   115.5   114.6   113.6
  114.25  113.53  114.03  113.22  113.14  112.88  110.27   109.5   111.9  111.94
   109.8  114.38  114.65  114.08  114.13   115.6   115.3   116.4     115   116.8
   116.7   115.7   115.3   116.6   118.3   117.2     117   113.6   113.3   115.8
     115   115.3   115.4   114.4     115   114.5   113.9   114.7   117.2   119.1
  -882.6  -752.6  -742.6  -732.6  -722.6  -672.6  -588.6   -98.6   261.4   761.4
   811.4   851.4   881.4   901.4  1001.4  1061.4  2641.4  2661.4  4094.1  4722.2
  4804.3  4804.7  4881.1  4924.6  4928.9  4943.1  4948.2 4952.31  4952.4 5030.49
  5030.6  5040.1  5068.4  5111.2  5279.4  5574.1  5894.1  5994.1  6054.1  6074.1
  6084.1  6094.1  6114.1  6134.1  6174.1  6194.1  6214.1  6254.1  6264.1  6304.1
  6494.1  6502.3  6612.3  6652.3  6732.3  6852.3  6892.3  7042.3  7092.3  7152.3
   122.3   121.1   121.4   120.9   119.8   118.2   118.5   117.1   117.4   116.7
   117.9   117.3     118   117.2   115.6   115.3   115.9   115.5   114.6   113.6
  114.26  114.07   114.1  113.23  114.15  114.18  114.19   114.2   114.2  114.24
  114.24  114.39  114.66  114.14  114.13   115.6   115.3   116.4     115   116.8
   116.7   115.7   115.3   116.6   118.3   117.2     117   113.6   113.3   115.8
     115   115.3   115.4   114.4     115   114.5   113.9   114.7   117.2   119.1
  122.25  121.05  121.35  120.85  119.75  118.15  118.45  117.05  117.35  116.65
  117.85  117.25  117.95  117.15  115.55  115.25  115.85  115.45  114.55  113.55
   114.2  113.48  113.98  113.17  113.09  112.83  110.22  109.45  111.85  111.89
  109.75  114.33   114.6  114.03  114.08  115.55  115.25  116.35  114.95  116.75
  116.65  115.65  115.25  116.55  118.25  117.15  116.95  113.55  113.25  115.75
  114.95  115.25  115.35  114.35  114.95  114.45  113.85  114.65  117.15  119.05
Pier Skew, UpSta & Num, DnSta & Num=  ,4971.7, 2 ,4971.7, 2 , 0 , 0 , 0 ,,
     1.4     1.4
  104.54  112.93
     1.4     1.4
  104.49  112.88
Pier Skew, UpSta & Num, DnSta & Num=  ,5018.2, 2 ,5018.2, 2 , 0 , 0 , 0 ,,
     1.4     1.4
  102.75  112.97
     1.4     1.4
   102.7  112.92
BR Coef= 1 , 1 , 0 ,1.25, 0 ,,,0.8,0,2,0,
WSPro=,,,, 1 ,,,, 0 ,,,, 0 ,,,,-1 ,-1 ,-1 , 0 , 0 , 0 , 0 , 0
BR U #Sta/Elev= 102
  -882.6   122.3  -752.6   121.1  -742.6   121.4  -732.6   120.9  -722.6   119.8
  -672.6   118.2  -588.6   118.5   -98.6   117.1   -48.6   117.2   261.4   117.4
   761.4   116.7   811.4   117.9   851.4   117.3   881.4     118   901.4   117.2
  1001.4   115.6  1061.4   115.3  1221.4   115.6  1379.2  115.63  2641.4   115.9
  2661.4   115.5  4094.1   114.6  4722.2   113.6  4723.5  113.67  4723.6  113.68
  4771.6  113.81  4774.7  113.85  4804.3  114.25  4804.7  113.53  4824.6  113.78
  4826.4  113.79  4881.1  114.03  4884.3  113.97  4924.4  113.23 4924.49  113.23
  4924.6  113.22 4924.71  113.22  4928.9  113.14  4943.1  112.88  4948.2  110.27
 4952.31   109.5  4952.4  109.48  4952.5  109.46  4971.7  105.86  4977.5  103.22
  4988.9  102.92  4990.3  101.11  4999.3  100.38  5004.6  102.93    5006   102.1
  5006.8  101.62  5011.1  103.15  5018.2  103.82  5030.4   109.7 5030.49  109.75
  5030.6   109.8  5040.1  114.38  5068.4  114.65 5070.09  114.63  5070.2  114.63
 5070.31  114.62  5111.2  114.08  5130.8  114.15  5187.9  114.34  5188.2  114.34
  5191.6  114.35    5248  114.13  5279.4  114.13  5574.1   115.6  5894.1   115.3
  5914.1   115.6  5934.1   115.9  5964.1   115.8  5994.1   116.4  6044.1   115.5
  6054.1     115  6074.1   116.8  6084.1   116.7  6094.1   115.7  6114.1   115.3
  6134.1   116.6  6174.1   118.3  6194.1   117.2  6214.1     117  6254.1   113.6
  6264.1   113.3  6304.1   115.8  6434.1   115.2  6494.1     115  6502.3   115.3
  6532.3     115  6582.3   115.2  6612.3   115.4  6652.3   114.4  6732.3     115
  6852.3   114.5  6892.3   113.9  7022.3   114.5  7042.3   114.7  7092.3   117.2
  7132.3   118.2  7152.3   119.1
BR U #Mann= 4
  -882.6      .2  1379.2     .14  4948.2    .035  5040.1     .14
BR U Banks=4948.2,5040.1
BR D #Sta/Elev= 102
  -882.6  122.25  -752.6  121.05  -742.6  121.35  -732.6  120.85  -722.6  119.75
  -672.6  118.15  -588.6  118.45   -98.6  117.05   -48.6  117.15   261.4  117.35
   761.4  116.65   811.4  117.85   851.4  117.25   881.4  117.95   901.4  117.15
  1001.4  115.55  1061.4  115.25  1221.4  115.55  1379.2  115.58  2641.4  115.85
  2661.4  115.45  4094.1  114.55  4722.2  113.55  4723.5  113.62  4723.6  113.63
  4771.6  113.76  4774.7   113.8  4804.3   114.2  4804.7  113.48  4824.6  113.73
  4826.4  113.74  4881.1  113.98  4884.3  113.92  4924.4  113.18 4924.49  113.18
  4924.6  113.17 4924.71  113.17  4928.9  113.09  4943.1  112.83  4948.2  110.22
 4952.31  109.45  4952.4  109.43  4952.5  109.41  4971.7  105.81  4977.5  103.17
  4988.9  102.87  4990.3  101.06  4999.3  100.33  5004.6  102.88    5006  102.05
  5006.8  101.57  5011.1   103.1  5018.2  103.77  5030.4  109.65 5030.49   109.7
  5030.6  109.75  5040.1  114.33  5068.4   114.6 5070.09  114.58  5070.2  114.58
 5070.31  114.57  5111.2  114.03  5130.8   114.1  5187.9  114.29  5188.2  114.29
  5191.6   114.3    5248  114.08  5279.4  114.08  5574.1  115.55  5894.1  115.25
  5914.1  115.55  5934.1  115.85  5964.1  115.75  5994.1  116.35  6044.1  115.45
  6054.1  114.95  6074.1  116.75  6084.1  116.65  6094.1  115.65  6114.1  115.25
  6134.1  116.55  6174.1  118.25  6194.1  117.15  6214.1  116.95  6254.1  113.55
  6264.1  113.25  6304.1  115.75  6434.1  115.15  6494.1  114.95  6502.3  115.25
  6532.3  114.95  6582.3  115.15  6612.3  115.35  6652.3  114.35  6732.3  114.95
  6852.3  114.45  6892.3  113.85  7022.3  114.45  7042.3  114.65  7092.3  117.15
  7132.3  118.15  7152.3  119.05
BR D #Mann= 4
  -882.6      .2  1379.2     .14  4948.2    .035  5040.1     .14
BR D Banks=4948.2,5040.1
BC Design=,, 0 ,, 0 ,,,,,,
BC HTab HWMax=122.29
BC Use User HTab Curves=0
BC User HTab FreeFlow(D)= 0

Type RM Length L Ch R = 1 ,209231.4,927.6,927.6,927.6
BEGIN DESCRIPTION:
Downstream Section of Bridge/Culvert/Weir
END DESCRIPTION:
XS GIS Cut Line= 6
      3064831.06     13914769.67      3064949.45      13914517.2
      3067444.11     13909651.28      3067509.77     13909517.33
      3067652.32     13909214.41      3068469.55     13907606.19
#Sta/Elev= 30
  -882.6  122.25  -742.6  121.35  -672.6  118.15   761.4  116.65   881.4  117.95
  1061.4  115.25  1379.2  115.58  4804.3   114.2  4943.1  112.83  4948.2  110.22
  4971.7  105.81  4977.5  103.17  4988.9  102.87  4990.3  101.06  4999.3  100.33
  5004.6  102.88  5006.8  101.57  5018.2  103.77  5040.1  114.33  5994.1  116.35
  6054.1  114.95  6074.1  116.75  6114.1  115.25  6174.1  118.25  6214.1  116.95
  6264.1  113.25  6304.1  115.75  6892.3  113.85  7042.3  114.65  7152.3  119.05
#Mann= 4 , 1 , 0
  -882.6      .2       0  1379.2     .14       0  4948.2    .035       0
  5040.1     .14       0
#XS Ineff= 2 , 0
       0    4837   118.5    5130       0   118.5
Permanent Ineff=
       F       F
Bank Sta=4948.2,5040.1
XS Rating Curve= 0 ,0
Exp/Cntr=0.5,0.3

Type RM Length L Ch R = 1 ,208303.8,712.7,746.7,824.6
BEGIN DESCRIPTION:
Cross Section 208303.8-Interpolated
END DESCRIPTION:
XS GIS Cut Line= 4
      3067404.01     13912073.75      3068299.61     13910244.03
      3068417.25     13909020.56       3068579.8     13907768.93
#Sta/Elev= 30
    2035   117.4    2725   116.3  4392.2   115.1  4842.2   113.8  4932.2     114
    4950  113.33  4975.3  104.89  4984.6  103.26  4992.2  100.67  5000.9     100
  5007.2  100.24  5007.8  100.94  5009.7  101.42  5020.6  102.94  5054.7  113.13
  5062.2   113.6  5132.2     114  5301.3   114.6  5481.3   114.9  5671.3   115.8
  5811.3   115.4  5961.3   115.7  6021.3   114.7  6071.3   115.3  6087.3  115.36
  6211.3   115.8  6311.8  116.55  6331.3   116.7  6521.3   116.9  6563.4   119.2
#Mann= 6 , 1 , 0
    2035     .14       0    4950    .035       0  5054.7     .14       0
  6087.3      .1       0  6311.8     .14       0  6563.4      .2       0
#XS Ineff= 2 , 0
       0                  5671.3       0   115.8
Permanent Ineff=
       F       F
Bank Sta=4950,5054.7
XS Rating Curve= 0 ,0
Exp/Cntr=0.3,0.1

Type RM Length L Ch R = 1 ,207557.1,659.7,703,708.2
BEGIN DESCRIPTION:
Cross Section 207557.1
END DESCRIPTION:
XS GIS Cut Line= 6
      3068614.63     13911085.03       3069040.1     13909903.19
      3069082.64     13909543.92       3069092.1     13909151.56
       3069092.1     13908924.65      3069145.51     13906640.98
#Sta/Elev= 30
  2926.3   116.8  3236.3   115.2  3806.3   115.4  4544.2   113.8  4914.4  110.94
    4950  112.56  4975.3  104.12  4984.6  102.49  4992.2    99.9  5000.9   99.23
  5007.2   99.47  5009.7  100.65  5020.6  102.17  5054.7  112.36  5102.2  112.02
  5126.7   114.5  5183.6   114.1  5613.6   115.3  5713.6     115  5755.7  116.05
  5773.6   116.5  5793.6   114.5    6216  118.08  6513.6     115  6833.6   115.7
  7113.6   115.3  7253.6   116.2  7403.6   115.1  7447.9   115.4    7448     119
#Mann= 5 , 1 , 0
  2926.3     .14       0    4950    .035       0  5054.7     .14       0
  5755.7      .1       0    6216      .2       0
#XS Ineff= 2 , 0
       0                  6213.6       0   118.1
Permanent Ineff=
       F       F
Bank Sta=4950,5054.7
XS Rating Curve= 0 ,0
Exp/Cntr=0.3,0.1

Type RM Length L Ch R = 1 ,206854.1,371.9,680.1,1180.7
BEGIN DESCRIPTION:
Cross Section 206854.1
END DESCRIPTION:
XS GIS Cut Line= 6
      3068427.88     13912085.32      3069096.82     13910654.83
      3069777.55     13909543.92      3069791.73     13909260.29
      3069782.27     13907898.84      3069705.73     13906370.79
#Sta/Elev= 30
  1722.9   117.6  2822.9   116.9  3672.1   114.1  3962.1   114.7  4592.1   112.8
    4635   114.2    4725   112.3    4865   113.5  4901.2  111.55  4953.5  112.92
  4976.1   104.6  4990.5  102.51  4999.2   98.71  5007.4  100.39  5041.8  101.86
  5060.7  111.87  5094.4  110.98  5127.3  112.37    5234   113.6    5364   113.8
    5424     118  5620.9   116.2  6080.9   116.5  6141.9   119.3  6570.5   114.9
  6860.5   113.5  6910.5   114.6  7390.5   114.4  7640.5     113  7780.5   116.7
#Mann= 4 , 1 , 0
  1722.9     .14       0  4953.5    .035       0  5060.7      .1       0
  6141.9      .2       0
#XS Ineff= 2 , 0
       0  3962.1   114.7  6141.9       0   119.3
Permanent Ineff=
       F       F
Bank Sta=4953.5,5060.7
XS Rating Curve= 0 ,0
Exp/Cntr=0.5,0.3

Type RM Length L Ch R = 1 ,206174.0,57,57,57
BEGIN DESCRIPTION:
Upstream Section of Bridge/Culvert/Weir
END DESCRIPTION:
XS GIS Cut Line= 5
       3068918.4     13911888.17      3069431.69     13910645.03
      3070896.61     13908448.67      3071174.98     13908016.19
      3070853.02     13905537.35
#Sta/Elev= 30
  1781.5   117.5  2481.5     117  2701.5   115.1  2791.5   117.3    2914  115.52
  3471.7   113.1  4724.4  114.87 4898.48  114.59 4936.61  113.22 4962.94  106.01
  4971.3  106.67  5004.1   98.64 5008.86   98.92 5014.43   105.2 5022.06  109.48
 5036.16  112.32 5043.79  112.08  5743.6   114.8  6183.6   113.5  6203.6   115.5
  6361.5  115.02  6530.5   111.8  6720.5   114.4  6780.5   112.3  6940.5   112.9
  7010.5   114.9  7490.5     113  8260.5   114.2  8520.5   114.9  8780.5   117.7
#Mann= 5 , 1 , 0
  1781.5      .1       0    2914     .14       0 4936.61    .035       0
 5043.79      .1       0  6361.5     .99       0
#XS Ineff= 2 , 0
       0    4920   115.6    5076       0   114.5
Permanent Ineff=
       F       F
Bank Sta=4936.61,5043.79
XS Rating Curve= 0 ,0
Exp/Cntr=0.5,0.3

Type RM Length L Ch R = 3 ,206145.5,,,
BEGIN DESCRIPTION:
CUTTEN ROAD - 35 degree skew
Structure ID: P00-80
END DESCRIPTION:
Bridge Culvert--1,0,-1,-1, 0
Deck Dist Width WeirC Skew NumUp NumDn MinLoCord MaxHiCord MaxSubmerge Is_Ogee
10,37,2.6,0, 60, 60, , , 0.95, 0, 1,1,,
  1781.5  2481.5  2701.5  2791.5    2914  2956.3  3076.3  3116.3  3186.3  3281.7
  3401.7  3471.7  3521.7  3591.7  3661.7  3920.8  3970.8  4200.8  4418.9    4631
  4664.4  4724.4  4828.6 4843.19  4843.3 4861.58 4898.48 4931.77 4931.86 5008.86
 5053.85 5053.96  5066.9 5067.01  5081.5 5134.32  5238.4 5320.87  5389.3  5653.6
  5743.6  5933.6  6113.6  6183.6  6203.6  6420.5  6480.5  6530.5  6590.5  6720.5
  6780.5  6860.5  6940.5  6990.5  7010.5  7490.5  8060.5  8260.5  8520.5  8780.5
   117.5   117.1   117.1  117.31  116.36  116.31  116.17  116.12  116.04  115.93
   115.9  115.85  115.47  115.36  115.28  115.04     115  114.96  115.04  115.11
  115.12  115.88   117.1  116.83  117.33  117.42  117.61  117.77  117.77  117.87
  117.82  117.82   117.8   117.3  117.28  116.23  114.23  114.02  113.84  114.09
  114.81  114.41  114.71  114.02  115.51  114.81  114.03  114.03  114.03  114.41
  114.04  114.04  114.05  114.05  114.91  114.07  114.61  114.21  114.91   117.7
   117.5     117   115.1   117.3  115.52   114.9   115.3   114.2   114.7   113.6
   114.1   113.1   113.3     113   113.5   113.2   113.6   113.9   113.4  113.77
  114.16  114.87  114.79  114.77  114.77  114.76  114.59  113.39  114.97  115.07
  115.02  112.08  112.08  112.08  112.08  112.08  112.81  113.32  112.92   113.6
   114.8   114.4   114.7   113.5   115.5   114.8   112.9   111.8   113.4   114.4
   112.3   113.6   112.9     114   114.9     113   114.6   114.2   114.9   117.7
  1781.5  2481.5  2701.5  2791.5    2914  2956.3  3076.3  3116.3  3186.3  3281.7
  3401.7  3471.7  3521.7  3591.7  3661.7  3920.8  3970.8  4200.8  4418.9    4631
  4664.4  4724.4  4828.6 4843.19  4843.3 4861.58 4898.48 4931.77 4931.86 5008.86
 5053.85 5053.96  5066.9 5067.01  5081.5 5134.32  5238.4 5320.87  5389.3  5653.6
  5743.6  5933.6  6113.6  6183.6  6203.6  6420.5  6480.5  6530.5  6590.5  6720.5
  6780.5  6860.5  6940.5  6990.5  7010.5  7490.5  8060.5  8260.5  8520.5  8780.5
   117.5   117.1   117.1  117.31  116.36  116.31  116.17  116.12  116.04  115.93
   115.9  115.85  115.47  115.36  115.28  115.04     115  114.96  115.04  115.11
  115.12  115.88   117.1  116.83  117.33  117.42  117.61  117.77  117.77  117.87
  117.82  117.82   117.8   117.3  117.28  116.23  114.23  114.02  113.84  114.09
  114.81  114.41  114.71  114.02  115.51  114.81  114.03  114.03  114.03  114.41
  114.04  114.04  114.05  114.05  114.91  114.07  114.61  114.21  114.91   117.7
  117.34  116.84  114.94  117.14  115.36  114.74  115.14  114.04  114.54  113.44
  113.94  112.94  113.14  112.84  113.34  113.04  113.44  113.74  113.24  113.61
     114  114.71  114.63  114.61  114.61   114.6  114.43  113.23  114.81  114.91
  114.86  111.92  111.92  111.92  111.92  111.92  112.65  113.16  112.76  113.44
  114.64  114.24  114.54  113.34  115.34  114.64  112.74  111.64  113.24  114.24
  112.14  113.44  112.74  113.84  114.74  112.84  114.44  114.04  114.74  117.54
Pier Skew, UpSta & Num, DnSta & Num=  ,4971.3, 2 ,4971.3, 2 , 0 , 0 , 0 ,,
     1.4     1.4
  105.51  116.04
     1.4     1.4
  105.35  115.88
Pier Skew, UpSta & Num, DnSta & Num=  ,5014.4, 2 ,5014.4, 2 , 0 , 0 , 0 ,,
     1.4     1.4
  103.41  116.06
     1.4     1.4
  103.25   115.9
Abutment Skew #Up #Dn= , 2 , 2
 4931.66 4962.94
  114.97  106.01
 4931.66 4962.94
  114.81  105.85
Abutment Skew #Up #Dn= , 2 , 2
 5018.53 5054.05
  106.88  115.02
 5018.53 5054.05
  106.72  114.86
BR Coef= 1 , 1 , 0 ,1.25, 0 ,,,0.8,-1,2,0,
WSPro=,,,, 1 ,,,, 0 ,,,, 0 ,,,,-1 ,-1 ,-1 , 0 , 0 , 0 , 0 , 0
BR U #Sta/Elev= 112
  1781.5   117.5  2171.5   117.3    2472  117.01  2481.5     117  2701.5   115.1
    2772  116.82  2791.5   117.3    2792  117.29    2914  115.52  2956.3   114.9
  3036.3   115.3  3076.3   115.3  3116.3   114.2  3186.3   114.7  3281.7   113.6
  3306.4  113.67  3351.7   113.8  3401.7   114.1  3416.4  113.89  3466.4  113.18
  3471.7   113.1  3506.4  113.24  3521.7   113.3  3591.7     113  3626.4  113.25
  3661.7   113.5  3776.4  113.28  3820.8   113.2  3920.8   113.2  3956.4  113.48
  3970.8   113.6  3976.4  113.61  4016.4  113.68  4080.8   113.8  4200.8   113.9
  4418.9   113.4    4631  113.77  4664.4  114.16  4724.4  114.87  4769.3  114.83
  4828.6  114.79 4843.19  114.77  4843.3  114.77 4843.41  114.77 4861.58  114.76
 4898.48  114.59 4931.77  113.39 4931.86  113.39 4936.61  113.22  4941.4  111.91
 4962.84  106.04 4962.94  106.01  4971.3  106.67 4990.41  102.22 4997.62   100.7
 4999.84   98.71  5004.1   98.64  5007.6   98.85 5008.86   98.92 5014.43   105.2
 5018.43  106.84 5018.53  106.88 5022.06  109.48 5036.16  112.32 5041.49  112.46
 5043.79  112.08 5053.85  112.08 5053.96  112.08 5066.79  112.08  5066.9  112.08
 5067.01  112.08  5081.5  112.08 5134.32  112.08 5156.54  112.31  5168.7  112.38
  5238.4  112.81 5320.87  113.32  5362.5   113.1  5389.3  112.92  5392.5   112.9
  5522.5   113.3  5636.4  113.56  5653.6   113.6  5743.6   114.8  5826.5  114.63
  5933.6   114.4  5993.6   114.5  6043.6   114.4  6113.6   114.7  6183.6   113.5
  6203.6   115.5  6270.5   115.4  6340.5   115.1  6361.5  115.02  6420.5   114.8
  6480.5   112.9  6530.5   111.8  6590.5   113.4  6720.5   114.4  6780.5   112.3
  6860.5   113.6  6940.5   112.9  6990.5     114  7010.5   114.9  7490.5     113
  7700.5   113.5  8060.5   114.6  8150.8  114.42  8260.5   114.2  8520.5   114.9
  8740.8  117.27  8780.5   117.7
BR U #Mann= 5
  1781.5      .1    2914     .14 4936.61    .035 5043.79      .1  6361.5     .99
BR U Banks=4936.61,5043.79
BR D #Sta/Elev= 112
  1781.5  117.34  2171.5  117.14    2472  116.85  2481.5  116.84  2701.5  114.94
    2772  116.66  2791.5  117.14    2792  117.13    2914  115.36  2956.3  114.74
  3036.3  115.14  3076.3  115.14  3116.3  114.04  3186.3  114.54  3281.7  113.44
  3306.4  113.51  3351.7  113.64  3401.7  113.94  3416.4  113.73  3466.4  113.02
  3471.7  112.94  3506.4  113.08  3521.7  113.14  3591.7  112.84  3626.4  113.09
  3661.7  113.34  3776.4  113.12  3820.8  113.04  3920.8  113.04  3956.4  113.32
  3970.8  113.44  3976.4  113.45  4016.4  113.52  4080.8  113.64  4200.8  113.74
  4418.9  113.24    4631  113.61  4664.4     114  4724.4  114.71  4769.3  114.67
  4828.6  114.63 4843.19  114.61  4843.3  114.61 4843.41  114.61 4861.58   114.6
 4898.48  114.43 4931.77  113.23 4931.86  113.23 4936.61  113.06  4941.4  111.75
 4962.84  105.88 4962.94  105.85  4971.3  106.51 4990.41  102.06 4997.62  100.54
 4999.84   98.55  5004.1   98.48  5007.6   98.69 5008.86   98.76 5014.43  105.04
 5018.43  106.68 5018.53  106.72 5022.06  109.32 5036.16  112.16 5041.49   112.3
 5043.79  111.92 5053.85  111.92 5053.96  111.92 5066.79  111.92  5066.9  111.92
 5067.01  111.92  5081.5  111.92 5134.32  111.92 5156.54  112.15  5168.7  112.22
  5238.4  112.65 5320.87  113.16  5362.5  112.94  5389.3  112.76  5392.5  112.74
  5522.5  113.14  5636.4   113.4  5653.6  113.44  5743.6  114.64  5826.5  114.47
  5933.6  114.24  5993.6  114.34  6043.6  114.24  6113.6  114.54  6183.6  113.34
  6203.6  115.34  6270.5  115.24  6340.5  114.94  6361.5  114.86  6420.5  114.64
  6480.5  112.74  6530.5  111.64  6590.5  113.24  6720.5  114.24  6780.5  112.14
  6860.5  113.44  6940.5  112.74  6990.5  113.84  7010.5  114.74  7490.5  112.84
  7700.5  113.34  8060.5  114.44  8150.8  114.26  8260.5  114.04  8520.5  114.74
  8740.8  117.11  8780.5  117.54
BR D #Mann= 5
  1781.5      .1    2914     .14 4936.61    .035 5043.79      .1  6361.5     .99
BR D Banks=4936.61,5043.79
BC Design=,, 0 ,, 0 ,,,,,,
BC HTab HWMax=117.7
BC Use User HTab Curves=0
BC User HTab FreeFlow(D)= 0

Type RM Length L Ch R = 1 ,206117.0,928.1,928.1,928.1
BEGIN DESCRIPTION:
Downstream Section of Bridge/Culvert/Weir
END DESCRIPTION:
XS GIS Cut Line= 5
      3068975.09     13911894.16      3069488.37     13910651.01
      3070953.29     13908454.65      3071231.66     13908022.17
      3070909.71     13905543.33
#Sta/Elev= 30
  1781.5  117.33  2481.5  116.83  2701.5  114.93  2791.5  117.13    2914  115.35
  3471.7  112.93  4724.4   114.7 4898.48  114.42 4936.61  113.05 4962.94  105.84
  4971.3   106.5  5004.1   98.47 5008.86   98.75 5014.43  105.03 5022.06  109.31
 5036.16  112.15 5043.79  111.91  5743.6  114.63  6183.6  113.33  6203.6  115.33
  6361.5  114.85  6530.5  111.63  6720.5  114.23  6780.5  112.13  6940.5  112.73
  7010.5  114.73  7490.5  112.83  8260.5  114.03  8520.5  114.73  8780.5  117.53
#Mann= 5 , 1 , 0
  1781.5      .1       0    2914     .14       0 4936.61    .035       0
 5043.79      .1       0  6361.5     .99       0
#XS Ineff= 2 , 0
       0    4920   114.7    5076       0     114
Permanent Ineff=
       F       F
Bank Sta=4936.61,5043.79
XS Rating Curve= 0 ,0
Exp/Cntr=0.5,0.3

Type RM Length L Ch R = 1 ,205188.9,680.6,444.8,340.5
BEGIN DESCRIPTION:
Cross Section 205188.9-Interpolated
END DESCRIPTION:
XS GIS Cut Line= 6
      3070936.08     13910737.51      3071019.93     13910545.69
      3071473.42     13909067.65      3071363.57     13908712.94
      3071330.78     13908398.32      3071109.47     13905185.98
#Sta/Elev= 30
    3010   116.2  3691.2  113.86  4239.3     113  4279.3   111.4  4399.3   113.8
  4579.3   113.7  4765.3   110.3  4865.3   111.7  4935.6  110.47    4956  104.44
  4972.4  102.62  4977.4   99.74  5003.5   97.75  5011.1  103.15  5019.6  104.25
  5038.1  110.89  5356.7   112.2  5386.7   114.8    5450  114.99    5653   112.6
    5913   113.1    6113   111.3    6463   113.1    6523   115.3    6573   113.7
    7093     113    8203   113.2    8513   114.9    8583     121    8673   123.7
#Mann= 5 , 1 , 0
    3010     .14       0  3691.2      .1       0  4935.6    .035       0
  5038.1      .1       0    5450      .2       0
#XS Ineff= 2 , 0
       0  3789.3   114.6    6523       0   115.3
Permanent Ineff=
       F       F
Bank Sta=4935.6,5038.1
XS Rating Curve= 0 ,0
Exp/Cntr=0.3,0.1

Type RM Length L Ch R = 1 ,204744.1,735.5,918.4,1216.1
BEGIN DESCRIPTION:
Cross Section 204744.1
END DESCRIPTION:
XS GIS Cut Line= 6
      3072268.62     13910301.32      3072192.85     13909732.64
      3072093.72     13909214.97       3071609.1     13908289.78
      3071487.94      13907452.7      3071400.88     13905024.25
#Sta/Elev= 30
  3186.2   114.8  3400.2   114.9  3610.2     111  3760.9   113.9    4528     111
    4658   112.9    4748     112    4808   108.8    4878   111.3  4935.6  110.06
    4956  104.03  4972.4  102.21  4977.4   99.33  5003.5   97.34  5011.1  102.74
  5019.6  103.84  5038.1  110.48  5119.1  110.51  5632.5   114.3  5982.5   113.3
  6022.5   111.7  6175.2  115.35  6268.3   113.6  6868.3   112.8  8008.3   112.1
  8428.3     114  8498.3   112.8  8518.3   113.8  8588.3   122.8  8608.3   129.9
#Mann= 5 , 1 , 0
  3186.2      .1       0  4935.6    .035       0  5038.1      .1       0
  5119.1     .14       0  6175.2      .2       0
#XS Ineff= 2 , 0
       0  3760.9   113.9  5662.5       0   114.3
Permanent Ineff=
       F       F
Bank Sta=4935.6,5038.1
XS Rating Curve= 0 ,0
Exp/Cntr=0.3,0.1

Type RM Length L Ch R = 1 ,203825.7,873,921.5,1022.5
BEGIN DESCRIPTION:
Cross Section 203825.7
Structure ID: PL1_P00-79_DSPL
END DESCRIPTION:
XS GIS Cut Line= 6
      3072675.76     13910611.88      3072802.93     13910070.73
      3072747.13     13908941.41      3072630.32     13908385.39
       3072578.5     13908126.31      3072442.26     13904767.31
#Sta/Elev= 30
  2558.9   115.3  2878.9   113.9  3114.8   114.4  3234.8   111.4  3394.8   114.2
  3574.8   111.7  3724.8   114.4  3914.8   111.7  4104.8   112.8  4355.5   109.4
  4535.5   108.5  4833.7   110.2 4953.29  109.78 4979.19  102.47 4987.29  101.74
 5000.99   95.49 5005.29   95.23 5010.59   95.34 5012.69   99.08 5048.09   110.7
  5257.9   110.1  5617.9   111.5  6167.9   111.8  6207.9   112.7  6227.9   111.1
  7537.9   111.7  7707.9     113  7926.6   113.1  8377.9   111.3  8439.6   113.5
#Mann= 4 , 1 , 0
  2558.9      .1       0 4953.29    .035       0 5048.09     .14       0
  7926.6     .99       0
#XS Ineff= 2 , 0
       0  3724.8   114.4  6207.9       0   112.7
Permanent Ineff=
       F       F
Bank Sta=4953.29,5048.09
XS Rating Curve= 0 ,0
Exp/Cntr=0.3,0.1

Type RM Length L Ch R = 1 ,202904.2,754.4,937.2,998.6
BEGIN DESCRIPTION:
Cross Section 202904.2
END DESCRIPTION:
XS GIS Cut Line= 6
      3073407.07     13909772.41      3073602.66     13909170.91
      3073602.66     13908818.46      3073492.52      13907838.2
      3073580.64     13906340.27       3073602.1     13904858.28
#Sta/Elev= 30
  3319.7  115.24  3439.7  112.27  3649.7  110.22  3669.7  111.76  3952.1  112.32
  4182.1   111.1  4292.1  111.89  4324.6   113.6  4440.1  111.58  4775.5  109.29
  4948.1  109.66  4992.9   96.21  4999.6   95.85    5028   98.13  5057.2  108.39
  5165.5  110.83  5284.5  110.99  5429.5   112.1  5563.6  110.03  6147.5  111.13
  6948.2  110.11  7004.6  112.88  7257.3  112.09  7377.3  113.58  7727.3   113.8
  7787.3  111.65  8217.3  109.73  8257.3  110.39  8267.3  114.06  8277.3  122.57
#Mann= 8 , 1 , 0
  3319.7      .1       0  4440.1     .14       0  4948.1    .035       0
  5057.2     .14       0  5284.5      .2       0  5429.5     .12       0
  6147.5     .14       0  6948.2      .1       0
#XS Ineff= 2 , 0
       0  4324.6   113.6  7004.6       0  112.88
Permanent Ineff=
       F       F
Bank Sta=4948.1,5057.2
XS Rating Curve= 0 ,0
Exp/Cntr=0.3,0.1

Type RM Length L Ch R = 1 ,201967.0,120.9,234,257.7
BEGIN DESCRIPTION:
Cross Section 201967.0-Interpolated
END DESCRIPTION:
XS GIS Cut Line= 6
      3073672.22     13909464.28      3073860.99     13908897.98
      3074399.21     13908395.54      3074466.65     13907836.57
      3074527.85     13907625.78      3074630.39      13904877.6
#Sta/Elev= 30
  3373.1   114.3  3503.1   113.7  3623.1     112  3893.1   112.5  3943.1   111.2
  4000.2  111.27    4420   109.5  4816.3   108.7  4856.3   110.8  4916.3   110.1
  4946.3   107.7 4954.85   107.6 4974.35  101.19 4990.85  100.16 4999.05   95.88
 5005.65      95 5009.35   95.38 5012.55   97.37 5016.75  101.06 5030.25  101.25
 5045.15  106.53  5056.3   107.3  5226.3   109.8  5269.4   108.9  6808.8   108.8
    6890  111.86    7689   111.5    8159   109.9    8229   110.4    8239   118.7
#Mann= 5 , 1 , 0
  3373.1      .1       0  4000.2     .14       0 4954.85    .035       0
 5045.15     .14       0    6890      .1       0
#XS Ineff= 2 , 0
       0                    6899       0   112.2
Permanent Ineff=
       F       F
Bank Sta=4954.85,5045.15
XS Rating Curve= 0 ,0
Exp/Cntr=0.3,0.1
