HEC-RAS study P100-00-00.prj: P100-00-00

--- P100-00-00.g01 (geometry) --- (continued)

Type RM Length L Ch R = 3 ,66051.7 ,,,
BEGIN DESCRIPTION:
GOLF COURSE BRIDGE1
Structure ID: P00-17
END DESCRIPTION:
Bridge Culvert--1,0,-1,-1, 0
Deck Dist Width WeirC Skew NumUp NumDn MinLoCord MaxHiCord MaxSubmerge Is_Ogee
10,13,2.6,0, 55, 55, , , 0.95, 0, 1,1,,
  2902.1  2982.1  3002.1  3162.1  3172.1  3252.1  3272.1  3372.1  3382.1  3482.1
  3522.1  3532.1  3572.1  3592.1  3602.1  3642.1  4270.9  4492.1  4582.1  4612.1
  4642.1  4662.1  4703.7    4782  4802.6  4924.4 4924.59  4924.7  4925.8  4981.2
  5022.5  5074.2 5074.31 5074.39  5074.5  5092.3  5120.7  5174.5    5227  5279.7
  5297.8  5337.8  5627.8  5647.8  5657.8  5667.8  6707.8  6727.8  6747.8  7257.8
  7558.7  7638.7  7658.7  7758.7  7888.7
   42.58   41.44   40.74   40.84   41.32   41.12   40.48   41.39   41.13   41.57
   41.14   40.47   41.42   41.39   40.81   40.95   39.25   40.37      38   37.88
   36.64   36.61   34.39   29.96   27.62   22.05   22.05   25.05    25.1   27.95
   27.78   25.01   22.01   22.01      22   21.09   20.98    23.6   31.28   34.65
   37.08   35.92   38.78   37.89   37.84   38.45   41.18   40.54   40.89   42.02
   42.47    42.4   41.08   41.31   43.41
   42.58   41.44   40.74   40.84   41.32   41.12   40.48   41.39   41.13   41.57
   41.14   40.47   41.42   41.39   40.81   40.95   39.25   40.37      38   37.88
   36.64   36.61   34.39   29.96   27.62   20.66   20.65   20.64    20.6   23.45
   23.28   20.51   20.51   20.51    20.2    20.5   20.98    23.6   31.28   34.65
   37.08   35.92   38.78   37.89   37.84   38.45   41.18   40.54   40.89   42.02
   42.47    42.4   41.08   41.31   43.41
  2902.1  2982.1  3002.1  3162.1  3172.1  3252.1  3272.1  3372.1  3382.1  3482.1
  3522.1  3532.1  3572.1  3592.1  3602.1  3642.1  4270.9  4492.1  4582.1  4612.1
  4642.1  4662.1  4703.7    4782  4802.6  4924.4 4924.59  4924.7  4925.8  4981.2
  5022.5  5074.2 5074.31 5074.39  5074.5  5092.3  5120.7  5174.5    5227  5279.7
  5297.8  5337.8  5627.8  5647.8  5657.8  5667.8  6707.8  6727.8  6747.8  7257.8
  7558.7  7638.7  7658.7  7758.7  7888.7
   42.58   41.44   40.74   40.84   41.32   41.12   40.48   41.39   41.13   41.57
   41.14   40.47   41.42   41.39   40.81   40.95   39.25   40.37      38   37.88
   36.64   36.61   34.39   29.96   27.62   22.05   22.05   25.05    25.1   27.95
   27.78   25.01   22.01   22.01      22   21.09   20.98    23.6   31.28   34.65
   37.08   35.92   38.78   37.89   37.84   38.45   41.18   40.54   40.89   42.02
   42.47    42.4   41.08   41.31   43.41
   42.54    41.4    40.7    40.8   41.28   41.08   40.44   41.35   41.09   41.53
    41.1   40.43   41.38   41.35   40.77   40.91   39.21   40.33   37.96   37.84
    36.6   36.57   34.35   29.92   27.58   20.62   20.61    20.6   20.56   23.41
   23.24   20.47   20.47   20.47   20.16   20.46   20.94   23.56   31.24   34.61
   37.04   35.88   38.74   37.85    37.8   38.41   41.14    40.5   40.85   41.98
   42.43   42.36   41.04   41.27   43.37
Pier Skew, UpSta & Num, DnSta & Num=  ,4964.5, 2 ,4964.5, 2 , 0 , 0 , 0 ,,
     1.3     1.3
      -1   23.62
     1.3     1.3
   -1.04   23.58
Pier Skew, UpSta & Num, DnSta & Num=  ,5034.6, 2 ,5034.6, 2 , 0 , 0 , 0 ,,
     1.3     1.3
    -.64   23.66
     1.3     1.3
    -.68   23.62
Abutment Skew #Up #Dn= , 2 , 2
  4924.6  4955.3
   20.64    9.15
  4924.6  4955.3
    20.6    9.11
Abutment Skew #Up #Dn= , 2 , 2
  5041.6 5074.59
    7.15   20.51
  5041.6 5074.59
    7.11   20.47
BR Coef= 1 , 1 , 0 ,1.25, 0 ,,,0.8,0,2,0,
WSPro=,,,, 1 ,,,, 0 ,,,, 0 ,,,,-1 ,-1 ,-1 , 0 , 0 , 0 , 0 , 0
BR U #Sta/Elev= 79
  2902.1   42.58  2982.1   41.44  3002.1   40.74  3162.1   40.84  3172.1   41.32
  3252.1   41.12  3272.1   40.48  3372.1   41.39  3382.1   41.13  3482.1   41.57
  3522.1   41.14  3532.1   40.47  3572.1   41.42    3592   41.39  3592.1   41.39
  3602.1   40.81  3642.1   40.95  4270.9   39.25  4272.1   39.25  4492.1   40.37
  4582.1      38  4612.1   37.88  4634.6   36.95  4642.1   36.64  4662.1   36.61
  4678.5   35.69  4703.7   34.39    4782   29.96  4802.6   27.62  4924.4   20.66
 4924.51   20.65 4924.59   20.65  4924.7   20.64  4924.8   20.64 4924.91   20.63
  4925.8   20.58  4955.2    9.26  4955.3    9.15  4962.1    1.49  4964.5     .07
  4968.5    -.38  4981.2   -1.81  4985.1   -2.25  4999.3   -3.85  5022.5    -.46
  5025.3    -.05  5034.6     .39  5037.9    1.42  5041.5       7  5041.6    7.15
  5071.3   20.15 5074.09    20.2  5074.2    20.2 5074.31    20.2 5074.39    20.2
  5074.5    20.2  5074.6   20.21  5092.3    20.5  5120.7   20.98  5174.5    23.6
    5227   31.28  5279.7   34.65  5297.8   37.08  5337.8   35.92  5627.8   38.78
  5647.8   37.89  5657.8   37.84  5667.8   38.45  6707.8   41.18  6727.8   40.54
  6747.8   40.89  7257.8   42.02  7352.8   42.16  7489.9   42.37  7558.7   42.47
  7638.7    42.4  7658.7   41.08  7758.7   41.31  7888.7   43.41
BR U #Mann= 8
  2902.1      .1    3592     .14  4270.9      .1  4634.6     .14  4925.8    .035
  5071.3      .1  7352.8     .14  7489.9      .2
BR U Banks=4925.8,5071.3
BR D #Sta/Elev= 79
  2902.1   42.54  2982.1    41.4  3002.1    40.7  3162.1    40.8  3172.1   41.28
  3252.1   41.08  3272.1   40.44  3372.1   41.35  3382.1   41.09  3482.1   41.53
  3522.1    41.1  3532.1   40.43  3572.1   41.38    3592   41.35  3592.1   41.35
  3602.1   40.77  3642.1   40.91  4270.9   39.21  4272.1   39.21  4492.1   40.33
  4582.1   37.96  4612.1   37.84  4634.6   36.91  4642.1    36.6  4662.1   36.57
  4678.5   35.65  4703.7   34.35    4782   29.92  4802.6   27.58  4924.4   20.62
 4924.51   20.61 4924.59   20.61  4924.7    20.6  4924.8    20.6 4924.91   20.59
  4925.8   20.54  4955.2    9.22  4955.3    9.11  4962.1    1.45  4964.5     .03
  4968.5    -.42  4981.2   -1.85  4985.1   -2.29  4999.3   -3.89  5022.5     -.5
  5025.3    -.09  5034.6     .35  5037.9    1.38  5041.5    6.96  5041.6    7.11
  5071.3   20.11 5074.09   20.16  5074.2   20.16 5074.31   20.16 5074.39   20.16
  5074.5   20.16  5074.6   20.17  5092.3   20.46  5120.7   20.94  5174.5   23.56
    5227   31.24  5279.7   34.61  5297.8   37.04  5337.8   35.88  5627.8   38.74
  5647.8   37.85  5657.8    37.8  5667.8   38.41  6707.8   41.14  6727.8    40.5
  6747.8   40.85  7257.8   41.98  7352.8   42.12  7489.9   42.33  7558.7   42.43
  7638.7   42.36  7658.7   41.04  7758.7   41.27  7888.7   43.37
BR D #Mann= 8
  2902.1      .1    3592     .14  4270.9      .1  4634.6     .14  4925.8    .035
  5071.3      .1  7352.8     .14  7489.9      .2
BR D Banks=4925.8,5071.3
BC Design=,, 0 ,, 0 ,,,,,,
BC HTab HWMax=43.41
BC Use User HTab Curves=0
BC User HTab FreeFlow(D)= 0

Type RM Length L Ch R = 1 ,66035.2 ,106.8,106.8,106.8
BEGIN DESCRIPTION:
Downstream Section of Bridge/Culvert/Weir
END DESCRIPTION:
XS GIS Cut Line= 4
      3164936.96     13872536.14      3163257.19     13873170.94
      3160909.45     13874805.82       3160698.2     13875059.33
#Sta/Elev= 30
  2902.1   42.78  3002.1   40.94  3272.1   40.68  3482.1   41.77  3532.1   40.67
    3592   41.59  4270.9   39.45  4492.1   40.57  4634.6   37.15  4703.7   34.59
  4925.8   20.78  4955.2    9.46  4962.1    1.69  4964.5     .27  4999.3   -3.65
  5037.9    1.62  5041.6    7.35  5071.3   20.35  5120.7   21.18  5174.5    23.8
    5227   31.48  5279.7   34.85  5297.8   37.28  5337.8   36.12  5627.8   38.98
  5657.8   38.04  7352.8   42.36  7489.9   42.57  7758.7   41.51  7888.7   43.61
#Mann= 8 , 1 , 0
  2902.1      .1       0    3592     .14       0  4270.9      .1       0
  4634.6     .14       0  4925.8    .035       0  5071.3      .1       0
  7352.8     .14       0  7489.9      .2       0
#XS Ineff= 2 , 0
       0    4915    21.1    5086       0      21
Permanent Ineff=
       F       F
Bank Sta=4925.8,5071.3
XS Rating Curve= 0 ,0
Exp/Cntr=0.5,0.3

Type RM Length L Ch R = 1 ,65928.4 ,711.7,840.8,937.6
BEGIN DESCRIPTION:
Cross Section 65928.4
END DESCRIPTION:
XS GIS Cut Line= 4
      3164615.09     13872471.88      3163083.77     13873136.64
      3162614.75     13873472.05      3160801.64     13874725.98
#Sta/Elev= 30
  3151.7    41.6  3431.7      39  3481.7    41.2    3840   39.78  4291.7    37.9
  4418.8   39.27  4621.7      40  4684.6   37.33  4741.7    35.9  4811.7    30.1
  4871.1    28.4  4891.1    25.5  4911.1    19.1  4921.6   17.74  4947.7   18.17
    4985    -.58  4996.4    -1.1  5015.3   -1.03  5060.9   18.83  5082.5   20.12
    5106   24.16  5151.1    25.1  5201.1    31.6  5261.1      35  5857.7    39.3
  6757.7    40.5  6857.7    43.5  6887.7    41.4  7275.4    41.9  7602.2    42.3
#Mann= 9 , 1 , 0
  3151.7      .2       0  3151.7      .1       0    3840     .14       0
  4418.8      .1       0  4684.6     .14       0  4947.7    .035       0
  5060.9      .1       0  7275.4     .14       0  7602.2      .2       0
Bank Sta=4947.7,5060.9
XS Rating Curve= 0 ,0
Exp/Cntr=0.3,0.1

Type RM Length L Ch R = 1 ,65087.6 ,1040.3,1038.9,949.1
BEGIN DESCRIPTION:
Cross Section 65087.6-Interpolated
END DESCRIPTION:
XS GIS Cut Line= 6
      3164555.08     13872398.54      3164001.66     13872478.55
      3163374.88     13872405.21      3162701.44     13872498.56
      3161981.31       13873152.      3161119.76     13874191.34
#Sta/Elev= 30
  3440.2    42.4  3620.2    39.6  3630.2    38.1  3670.2    40.4  3690.2    39.3
  4319.4    39.7  4419.4    35.5  4658.6    34.2  4750.4    30.3  4800.4    18.7
  4830.4    15.7  4912.3   20.33  4966.2    7.32  4977.5    3.92  4980.5     .48
  4987.8   -2.49  4995.4      -4  5019.8    1.36  5028.6    7.97  5059.2   16.82
  5130.4    22.1  5180.4    30.5  5300.4    35.6  5720.3    33.9  5920.3    38.1
  6602.7    37.6  6642.5   36.22  6662.7    38.5  6702.7      39  7632.7    41.6
#Mann= 6 , 1 , 0
  3440.2      .2       0  3440.2      .1       0  4658.6     .14       0
  4912.3    .035       0  5059.2     .14       0  6642.5      .1       0
Bank Sta=4912.3,5059.2
XS Rating Curve= 0 ,0
Exp/Cntr=0.3,0.1

Type RM Length L Ch R = 1 ,64048.7 ,197.1,516.2,867.9
BEGIN DESCRIPTION:
Cross Section 64048.7
END DESCRIPTION:
XS GIS Cut Line= 6
      3164761.39     13871946.73      3162826.62     13871745.97
        3162468.     13871745.97       3162050.7      13871948.1
      3161842.05     13872561.02      3160749.88     13874377.98
#Sta/Elev= 30
  2480.2    41.2  2920.2    39.2  3730.1    39.3  4010.1    35.2  4060.1    31.3
  4100.1    32.4  4190.1      29  4393.8   27.48  4445.7    26.6  4485.7    18.5
  4565.7    16.5  4635.7    22.1  4705.7      17  4755.7      19  4864.3    18.5
  4872.5   21.08  4912.3   21.91  4977.5     1.5  4980.5   -1.94  4995.4   -6.42
  5019.8   -1.06  5028.6    5.55  5059.2    14.4  5091.3   18.14  5164.3    20.9
  5194.3    28.8    5248    33.3  7145.6   39.64  7553.2    40.6  8015.4    43.5
#Mann= 7 , 1 , 0
  2480.2      .2       0  2480.2      .1       0  4393.8     .14       0
  4912.3    .035       0  5059.2     .14       0  7145.6      .1       0
  7553.2     .14       0
Bank Sta=4912.3,5059.2
XS Rating Curve= 0 ,0
Exp/Cntr=0.3,0.1

Type RM Length L Ch R = 1 ,63532.5 ,129,178.1,179.2
BEGIN DESCRIPTION:
Cross Section 63532.5-Interpolated
END DESCRIPTION:
XS GIS Cut Line= 6
       3164498.1     13871903.01      3163553.71     13871822.97
      3162930.67     13871729.09      3162388.72     13871455.98
      3161974.78     13871003.63      3161680.33     13870832.94
#Sta/Elev= 30
    2692    41.5  2858.9      39  3278.9    39.9  3769.8      38  3966.7    34.7
  3996.7      32  4036.7    32.7  4126.7    28.8  4329.3   27.71  4409.9    27.6
  4479.9    29.8  4665.8    31.5  4689.8    29.3  4793.4   24.66  4815.8    25.1
  4906.9    17.1  4926.9    17.5  4934.6   12.35  4973.7      -2  4999.8      -3
  5028.8   -1.14  5058.3   11.76  5066.9      10  5088.1    12.3  5138.1    14.4
  5198.1    28.4  5490.3    38.5  5620.3    39.8  5680.3    38.8  5830.7      41
#Mann= 7 , 1 , 0
    2692      .1       0  4329.3     .14       0  4689.8      .1       0
  4793.4     .14       0  4934.6    .035       0  5058.3     .14       0
  5830.7      .2       0
Bank Sta=4934.6,5058.3
XS Rating Curve= 0 ,0
Exp/Cntr=0.5,0.3

Type RM Length L Ch R = 1 ,63354.4 ,30,30,30
BEGIN DESCRIPTION:
Upstream Section of Bridge/Culvert/Weir
END DESCRIPTION:
XS GIS Cut Line= 6
      3164536.01     13871806.03      3163194.57     13871724.21
      3163072.53     13871688.13      3162709.86     13871518.67
       3162136.6     13870941.54      3161925.14     13870779.91
#Sta/Elev= 30
  2734.6   40.57  2904.6   38.97  3614.6   38.87  3714.6   37.37  3734.6   38.47
  3852.3   36.87  3942.3   33.07  3982.3   34.87  4052.3   31.67  4102.3   32.37
  4210.5   28.07  4350.5   26.67  4538.2   30.37  4600.1   33.63  4683.6   31.96
  4839.4    30.7  4879.1   15.16  4934.6   12.95  4961.1    4.65  4973.7    -1.4
  4999.8    -2.4  5028.8    -.54  5058.3   12.36    5076   11.14  5137.8   31.16
  5149.3   29.81  5219.8    32.1  5495.1   37.78  5668.4   38.87  5688.4   40.17
#Mann= 7 , 1 , 0
  2734.6     .14       0  4683.6      .1       0  4839.4     .14       0
  4934.6    .035       0  5058.3     .14       0  5219.8      .1       0
  5495.1     .14       0
#XS Ineff= 2 , 0
       0    4831      32    5147       0      35
Permanent Ineff=
       F       F
Bank Sta=4934.6,5058.3
XS Rating Curve= 0 ,0
Exp/Cntr=0.5,0.3

Type RM Length L Ch R = 3 ,63339.4 ,,,
BEGIN DESCRIPTION:
GREEN RIVER (LEY) ROAD
Structure ID: P00-16A
END DESCRIPTION:
Bridge Culvert--1,0,-1,-1, 0
Deck Dist Width WeirC Skew NumUp NumDn MinLoCord MaxHiCord MaxSubmerge Is_Ogee
10,10,2.6,0, 60, 60, , , 0.95, 0, 1,1,,
  2734.6  2874.6  2904.6  3204.6  3494.6  3614.6  3664.6  3714.6  3734.6  3772.3
  3812.3  3852.3  3872.3  3882.3  3892.3  3922.3  3932.3  3942.3  3952.3  3962.3
  3982.3  4032.3  4052.3  4082.3  4102.3  4172.3  4180.5  4190.5  4210.5  4350.5
  4418.2  4438.2  4538.2  4568.1  4572.1  4600.1  4674.2  4698.2 4752.99  4753.1
 4841.11  4841.2 5136.79  5136.9  5137.8  5149.3  5175.7  5277.9  5313.8 5313.91
  5359.9  5391.7  5416.2  5470.9  5490.9  5500.9  5538.4  5568.4  5668.4  5688.4
    40.6      40      39    39.4    38.8   38.91   38.51   37.41   38.51   38.11
   36.51   36.91   35.51   35.91   35.21   34.71   33.51   33.11   33.51   34.81
   34.91   33.31   32.04   32.31   32.41   32.09   32.09   32.09   32.11   32.26
   32.34   32.36   32.37   32.78   33.07   33.67   33.93    34.2   34.71   37.21
   37.84   37.84   37.83   37.83   37.83   37.84   37.87   37.29   37.43   35.05
   35.74   36.68   37.11    37.7    37.6    38.1    38.4    38.2    38.9    40.2
    40.6      40      39    39.4    38.8    38.9    38.5    37.4    38.5    38.1
    36.5    36.9    35.5    35.9    35.2    34.7    33.5    33.1    33.5    34.8
    34.9    33.3    31.7    32.3    32.4    29.1    29.1    29.5    28.1    26.7
    27.9    29.2    30.4   32.73   33.06   33.66   32.62   31.01   30.86   30.86
    30.6   32.44   32.43    30.9   31.19   29.84    30.7      34   35.04   35.04
   35.74   36.68   37.11    37.7    37.6    38.1    38.4    38.2    38.9    40.2
  2734.6  2874.6  2904.6  3204.6  3494.6  3614.6  3664.6  3714.6  3734.6  3772.3
  3812.3  3852.3  3872.3  3882.3  3892.3  3922.3  3932.3  3942.3  3952.3  3962.3
  3982.3  4032.3  4052.3  4082.3  4102.3  4172.3  4180.5  4190.5  4210.5  4350.5
  4418.2  4438.2  4538.2  4568.1  4572.1  4600.1  4674.2  4698.2 4752.99  4753.1
 4841.11  4841.2 5136.79  5136.9  5137.8  5149.3  5175.7  5277.9  5313.8 5313.91
  5359.9  5391.7  5416.2  5470.9  5490.9  5500.9  5538.4  5568.4  5668.4  5688.4
    40.6      40      39    39.4    38.8   38.91   38.51   37.41   38.51   38.11
   36.51   36.91   35.51   35.91   35.21   34.71   33.51   33.11   33.51   34.81
   34.91   33.31   32.04   32.31   32.41   32.09   32.09   32.09   32.11   32.26
   32.34   32.36   32.37   32.78   33.07   33.67   33.93    34.2   34.71   37.21
   37.84   37.84   37.83   37.83   37.83   37.84   37.87   37.29   37.43   35.05
   35.74   36.68   37.11    37.7    37.6    38.1    38.4    38.2    38.9    40.2
   40.54   39.94   38.94   39.34   38.74   38.84   38.44   37.34   38.44   38.04
   36.44   36.84   35.44   35.84   35.14   34.64   33.44   33.04   33.44   34.74
   34.84   33.24   31.64   32.24   32.34   29.04   29.04   29.44   28.04   26.64
   27.84   29.14   30.34   32.67      33    33.6   32.56   30.95    30.8    30.8
   30.54   32.38   32.37   30.84   31.13   29.78   30.64   33.94   34.98   34.98
   35.68   36.62   37.05   37.64   37.54   38.04   38.34   38.14   38.84   40.14
Pier Skew, UpSta & Num, DnSta & Num=  ,4900.4, 2 ,4900.4, 2 , 0 , 0 , 0 ,,
     2.4     2.4
   13.69   33.44
     2.4     2.4
   13.63   33.38
Pier Skew, UpSta & Num, DnSta & Num=  ,4961.1, 2 ,4961.1, 2 , 0 , 0 , 0 ,,
     2.4     2.4
    2.83   33.44
     2.4     2.4
    2.77   33.38
Pier Skew, UpSta & Num, DnSta & Num=  ,5018.8, 2 ,5018.8, 2 , 0 , 0 , 0 ,,
     2.4     2.4
   -2.39   33.43
     2.4     2.4
   -2.45   33.37
Pier Skew, UpSta & Num, DnSta & Num=  ,5079, 2 ,5079, 2 , 0 , 0 , 0 ,,
     2.4     2.4
    10.7   33.43
     2.4     2.4
   10.64   33.37
BR Coef= 1 , 1 , 0 ,1.25, 0 ,,,0.8,0,2,0,
WSPro=,,,, 1 ,,,, 0 ,,,, 0 ,,,,-1 ,-1 ,-1 , 0 , 0 , 0 , 0 , 0
BR U #Sta/Elev= 104
  2734.6    40.6  2874.6      40  2904.6      39  3204.6    39.4  3494.6    38.8
  3537.2   38.84  3614.6    38.9  3664.6    38.5  3714.6    37.4  3734.6    38.5
  3772.3    38.1  3812.3    36.5  3852.3    36.9  3872.3    35.5  3882.3    35.9
  3892.3    35.2  3922.3    34.7  3932.3    33.5  3942.3    33.1  3952.3    33.5
  3957.2   34.14  3962.3    34.8  3982.3    34.9  4002.3    34.2  4032.3    33.3
  4052.3    31.7  4082.3    32.3  4102.3    32.4  4172.3    29.1  4180.5    29.1
  4190.5    29.5  4205.9   28.42  4210.5    28.1  4350.5    26.7  4358.2    26.9
  4418.2    27.9  4438.2    29.2  4473.3   29.62  4533.3   30.34  4538.2    30.4
  4545.6    30.9  4568.1   32.73  4572.1   33.06  4600.1   33.66  4657.2   32.86
  4674.2   32.62  4683.6   31.99  4698.2   31.01  4726.9   30.92    4742   30.88
 4752.99   30.86  4753.1   30.86 4753.21   30.86  4831.9   30.74  4839.4   30.73
  4840.8   30.73    4841   30.65 4841.11    30.6  4841.2   30.57  4841.8   30.32
  4857.3   24.03  4879.1   15.19  4885.8    14.2  4900.4   14.78  4912.1   13.87
  4934.6   12.98  4961.1    4.68  4965.7    1.43  4973.7   -1.37  4999.8   -2.37
  5018.8   -1.32  5028.8    -.51  5034.4    1.42  5058.3   12.39    5076   11.17
    5079   12.06  5108.1   21.65  5136.7   30.84 5136.79   30.87  5136.9    30.9
    5137   30.93  5137.8   31.19  5149.3   29.84  5175.7    30.7  5217.3   32.05
  5219.8   32.13  5227.3   32.37  5277.9      34  5307.3   34.94 5313.69   35.04
  5313.8   35.04 5313.91   35.04  5333.2   35.33  5359.9   35.74  5391.7   36.68
  5416.2   37.11  5470.9    37.7  5490.9    37.6  5495.1   37.81  5500.9    38.1
  5538.4    38.4  5568.4    38.2  5668.4    38.9  5688.4    40.2
BR U #Mann= 7
  2734.6     .14  4683.6      .1  4839.4     .14  4934.6    .035  5058.3     .14
  5219.8      .1  5495.1     .14
BR U Banks=4934.6,5058.3
BR D #Sta/Elev= 104
  2734.6   40.54  2874.6   39.94  2904.6   38.94  3204.6   39.34  3494.6   38.74
  3537.2   38.78  3614.6   38.84  3664.6   38.44  3714.6   37.34  3734.6   38.44
  3772.3   38.04  3812.3   36.44  3852.3   36.84  3872.3   35.44  3882.3   35.84
  3892.3   35.14  3922.3   34.64  3932.3   33.44  3942.3   33.04  3952.3   33.44
  3957.2   34.08  3962.3   34.74  3982.3   34.84  4002.3   34.14  4032.3   33.24
  4052.3   31.64  4082.3   32.24  4102.3   32.34  4172.3   29.04  4180.5   29.04
  4190.5   29.44  4205.9   28.36  4210.5   28.04  4350.5   26.64  4358.2   26.84
  4418.2   27.84  4438.2   29.14  4473.3   29.56  4533.3   30.28  4538.2   30.34
  4545.6   30.84  4568.1   32.67  4572.1      33  4600.1    33.6  4657.2    32.8
  4674.2   32.56  4683.6   31.93  4698.2   30.95  4726.9   30.86    4742   30.82
 4752.99    30.8  4753.1    30.8 4753.21    30.8  4831.9   30.68  4839.4   30.67
  4840.8   30.67    4841   30.59 4841.11   30.54  4841.2   30.51  4841.8   30.26
  4857.3   23.97  4879.1   15.13  4885.8   14.14  4900.4   14.72  4912.1   13.81
  4934.6   12.92  4961.1    4.62  4965.7    1.37  4973.7   -1.43  4999.8   -2.43
  5018.8   -1.38  5028.8    -.57  5034.4    1.36  5058.3   12.33    5076   11.11
    5079      12  5108.1   21.59  5136.7   30.78 5136.79   30.81  5136.9   30.84
    5137   30.87  5137.8   31.13  5149.3   29.78  5175.7   30.64  5217.3   31.99
  5219.8   32.07  5227.3   32.31  5277.9   33.94  5307.3   34.88 5313.69   34.98
  5313.8   34.98 5313.91   34.98  5333.2   35.27  5359.9   35.68  5391.7   36.62
  5416.2   37.05  5470.9   37.64  5490.9   37.54  5495.1   37.75  5500.9   38.04
  5538.4   38.34  5568.4   38.14  5668.4   38.84  5688.4   40.14
BR D #Mann= 7
  2734.6     .14  4683.6      .1  4839.4     .14  4934.6    .035  5058.3     .14
  5219.8      .1  5495.1     .14
BR D Banks=4934.6,5058.3
BC Design=,, 0 ,, 0 ,,,,,,
BC HTab HWMax=40.57
BC Use User HTab Curves=0
BC User HTab FreeFlow(D)= 0

Type RM Length L Ch R = 1 ,63324.4 ,1228.6,1228.6,1228.6
BEGIN DESCRIPTION:
Downstream Section of Bridge/Culvert/Weir
END DESCRIPTION:
XS GIS Cut Line= 6
       3164557.5     13871785.09      3163216.05     13871703.27
      3163094.01     13871667.19      3162731.34     13871497.73
      3162158.08      13870920.6      3161946.63     13870758.98
#Sta/Elev= 30
  2734.6    40.5  2904.6    38.9  3614.6    38.8  3714.6    37.3  3734.6    38.4
  3852.3    36.8  3942.3      33  3982.3    34.8  4052.3    31.6  4102.3    32.3
  4210.5      28  4350.5    26.6  4538.2    30.3  4600.1   33.56  4683.6   31.89
  4839.4   30.63  4879.1   15.09  4934.6   12.88  4961.1    4.58  4973.7   -1.47
  4999.8   -2.47  5028.8    -.61  5058.3   12.29    5076   11.07  5137.8   31.09
  5149.3   29.74  5219.8   32.03  5495.1   37.71  5668.4    38.8  5688.4    40.1
#Mann= 7 , 1 , 0
  2734.6     .14       0  4683.6      .1       0  4839.4     .14       0
  4934.6    .035       0  5058.3     .14       0  5219.8      .1       0
  5495.1     .14       0
#XS Ineff= 2 , 0
       0    4831    31.8    5147       0    34.8
Permanent Ineff=
       F       F
Bank Sta=4934.6,5058.3
XS Rating Curve= 0 ,0
Exp/Cntr=0.5,0.3

Type RM Length L Ch R = 1 ,62095.8 ,997.7,995.5,867.1
BEGIN DESCRIPTION:
Cross Section 62095.8
END DESCRIPTION:
XS GIS Cut Line= 5
      3165280.35     13871395.19      3163616.86     13870515.27
      3163126.56     13870265.85      3161676.99     13869659.13
      3161539.42     13869492.59
#Sta/Elev= 30
  2797.8   41.22  3045.8   38.32  4341.8   36.01  4373.8   38.29  4397.8   36.67
  4439.6   40.72  4541.8   35.72  4629.8   39.75  4669.8   31.66  4799.7   23.38
  4815.7    14.5  4839.7   10.25  4903.7   16.79  4938.3   15.36  4985.2   -6.18
    5025   -7.77  5028.6     .33  5050.8   12.76    5144   10.22  5177.1   17.57
    5201   22.87  5253.8   26.41  5269.8   19.79  5301.8   13.79  5662.9   13.67
  6749.8   13.29  6809.2   16.92  6905.2   39.62  6977.2   40.45  7017.2   44.96
#Mann= 6 , 1 , 0
  2797.8      .1       0  4439.6     .14       0  4938.3    .035       0
  5050.8     .12       0  5177.1     .08       0  5662.9      .2       0
Bank Sta=4938.3,5050.8
XS Rating Curve= 0 ,0
Exp/Cntr=0.3,0.1

Type RM Length L Ch R = 1 ,61100.3 ,1102.1,1092.7,1058.1
BEGIN DESCRIPTION:
Cross Section 61100.3
END DESCRIPTION:
XS GIS Cut Line= 6
      3165769.52     13870656.92      3164976.04     13869900.64
       3163843.8     13869587.73      3163563.42     13869444.29
      3163178.72     13869431.25       3163038.8     13869372.05
#Sta/Elev= 30
    2324   40.32  2577.3   38.39    2652   38.41    2676   35.62    2716   38.55
    3180   37.01    3316   38.64  3460.2   36.41  3732.2   37.23  4439.5   27.06
  4492.1   26.29  4508.1   23.05  4556.1   20.89  4682.8   18.32  4738.8   13.32
  4805.4   12.42  4837.4    8.96  4940.4   13.12  4970.2     .28  4971.4   -2.62
    4975   -4.22  4990.9   -8.68  5027.6   -1.52  5073.5   17.64  5168.2   10.23
  5177.1   13.08  5228.7   29.58  5285.8   32.44  5342.7   37.92  5446.7   52.45
#Mann= 6 , 1 , 0
    2324      .2       0  2577.3      .1       0  4439.5     .14       0
  4940.4    .035       0  5073.5     .12       0  5177.1     .08       0
Bank Sta=4940.4,5073.5
XS Rating Curve= 0 ,0
Exp/Cntr=0.3,0.1

Type RM Length L Ch R = 1 ,60007.6 ,1174,1126.4,990.9
BEGIN DESCRIPTION:
Cross Section 60007.6
END DESCRIPTION:
XS GIS Cut Line= 6
      3166266.72     13870399.04      3165577.33     13869515.98
      3163993.76     13868746.61      3163335.21       13868551.
      3163126.56     13868511.88      3162819.95     13868280.67
#Sta/Elev= 30
  1190.6   39.21  1222.6   37.02  1369.7   38.07  3190.9   35.99  3334.9   37.11
  3462.9   35.58  3846.9   36.12  3958.9   34.67  4054.9   36.39  4079.4   40.24
  4095.4   40.87  4203.7   36.32  4319.4   37.11  4578.5   31.75  4758.7   29.81
  4800.7   27.94  4830.7   17.86  4870.7    9.62  4955.7    9.23  4972.6     .44
  4974.6   -2.18  4995.1   -7.78  5025.3    -1.1  5071.9   14.77    5101    13.5
  5130.5   12.21  5193.4   33.67    5235   33.89    5267   40.36    5355   53.12
#Mann= 8 , 1 , 0
  1190.6      .2       0  1369.7      .1       0  4203.7     .14       0
  4578.5      .1       0  4800.7     .14       0  4955.7    .035       0
  5071.9     .12       0    5101     .08       0
Bank Sta=4955.7,5071.9
XS Rating Curve= 0 ,0
Exp/Cntr=0.3,0.1

Type RM Length L Ch R = 1 ,58881.2 ,295.9,388.6,405.9
BEGIN DESCRIPTION:
Cross Section 58881.2
END DESCRIPTION:
XS GIS Cut Line= 5
      3166711.77     13870483.35      3166157.89     13869130.62
      3164202.42     13867651.19      3163798.15     13867501.22
      3163150.22      13867490.6
#Sta/Elev= 30
   367.1   38.77   780.2   38.08  2476.8   34.43  2500.8   36.63  2876.8   36.12
  2932.8   33.91  2956.8    35.8  3404.8   37.73  3772.8   34.31  4280.9   34.52
  4523.6   31.39  4760.1   25.73  4792.1   21.82  4808.1   14.96  4832.1   18.93
  4896.1   10.59  4941.8   11.33  4966.8    2.64  4970.5     .32  4975.1   -6.71
  4998.8   -9.53  5027.3   -1.79  5039.6    6.76  5056.2    11.9  5129.7    9.05
    5154   16.04  5204.9   30.67  5248.1   30.23  5320.1   43.84  5360.1   54.57
#Mann= 6 , 1 , 0
   367.1      .2       0   780.2      .1       0  4523.6     .14       0
  4941.8    .035       0  5056.2     .12       0    5154     .08       0
Bank Sta=4941.8,5056.2
XS Rating Curve= 0 ,0
Exp/Cntr=0.3,0.1

Type RM Length L Ch R = 1 ,58492.6 ,439.9,501.4,529.6
BEGIN DESCRIPTION:
Cross Section 58492.6-Interpolated
END DESCRIPTION:
XS GIS Cut Line= 6
      3167976.96     13869986.11      3166505.81     13868777.45
      3165208.55     13867930.22      3163623.45     13867119.61
      3163311.58     13867082.48      3163175.64     13867082.48
#Sta/Elev= 30
    -328   38.94   316.6   38.16   659.8   38.02  2167.9   34.57  2327.9    36.7
  2575.9   34.73  2599.9   36.66  2631.9   34.78  3023.9   33.86  3557.4   36.49
  3927.6   33.87  4043.1   34.16    4298   31.23  4639.8   26.02  4735.8   22.47
  4799.8   11.86  4815.8   16.99  4831.8   17.99  4905.4    9.97  4954.8   -1.14
  5007.5      -9    5026   -8.68  5045.2    -.99  5053.1     8.2  5057.8   10.84
  5124.6    9.87  5201.8   31.15  5227.8    30.1  5283.8   36.68  5355.8   53.34
#Mann= 9 , 1 , 0
    -328      .2       0   316.6     .14       0   659.8      .1       0
  3927.6     .14       0  4043.1      .1       0    4298     .14       0
  4905.4    .035       0  5053.1     .12       0  5124.6     .08       0
Bank Sta=4905.4,5053.1
XS Rating Curve= 0 ,0
Exp/Cntr=0.5,0.3

Type RM Length L Ch R = 1 ,57991.2 ,54,54,54
BEGIN DESCRIPTION:
Upstream Section of Bridge/Culvert/Weir
END DESCRIPTION:
XS GIS Cut Line= 6
      3168969.09     13869426.83      3165559.84     13867624.28
      3164374.28     13866990.56      3163924.97     13866746.54
      3163444.68     13866510.26      3161948.23     13865710.43
#Sta/Elev= 30
  -964.4   38.62   -47.4   37.63    1954   34.93    2674   35.55    2722   38.69
  2780.5   35.87  3052.5   36.89  3148.5   34.23  3862.7   35.77    4401   27.94
    4497   21.85    4545   25.31  4546.5   22.85  4783.8   22.33  4799.5   21.94
  4830.8    13.2  4905.4   10.15  5007.5   -6.82    5026    -6.5  5045.2    1.19
  5053.1    8.38  5106.5   15.42  5115.5   14.29  5139.1   20.39  5200.4   27.21
    5262   25.42  5518.4   29.49  5736.2   33.14  6784.2    34.9  6979.7   38.91
#Mann= 5 , 1 , 0
  -964.4      .2       0   -47.4      .1       0  4905.4    .035       0
  5053.1      .1       0  5518.4     .08       0
#XS Ineff= 2 , 0
       0    4775    34.8    5169       0    34.9
Permanent Ineff=
       F       F
Bank Sta=4905.4,5053.1
XS Rating Curve= 0 ,0
Exp/Cntr=0.5,0.3

Type RM Length L Ch R = 3 ,57964.2 ,,,
BEGIN DESCRIPTION:
SOUTHERN PACIFIC RAILROAD
Structure ID: P00-16
END DESCRIPTION:
Bridge Culvert--1,0,-1,-1, 0
Deck Dist Width WeirC Skew NumUp NumDn MinLoCord MaxHiCord MaxSubmerge Is_Ogee
10,34,2.6,0, 60, 60, , , 0.95, 0, 1,1,,
  -964.4  -188.4   955.6  1035.6  1059.6  1083.6    1130    1346    1378    1506
    1538    1554    2674    2722  2780.5  2916.5  2972.5  3020.5  3052.5  3148.5
  3862.7  4006.7  4078.7    4401    4449    4497    4545  4546.5 4785.21  4785.3
 5159.29  5159.4  5200.4    5214    5230    5262    5278    5342  5472.2  5488.2
  5568.2  5608.2  5656.2  5696.2  5736.2  5768.2  5872.2  5888.2  5952.2  6120.2
  6176.2  6344.2  6496.2  6592.2  6624.2  6640.2  6688.2  6864.2  6928.2  6979.7
   38.66   37.16   37.36   36.66   37.43   35.68   36.53   36.36   37.26   36.58
   34.87   35.53   35.59   38.73   35.92    35.9   36.91    35.9   36.94    35.9
   35.82   35.69   35.67   35.57   35.55   35.54   35.52   35.52   35.54   35.54
    35.4    35.4   35.36   35.35   35.34   35.31    35.3   35.31   35.36   35.37
    35.4   35.42   35.44   35.45   35.47   35.48   35.53   35.53   35.56   35.63
   35.65   35.72   35.78    35.8    35.8    35.8    35.8    35.8   36.37   38.95
   38.66   37.16   37.36   36.66   37.43   35.68   36.53   36.36   37.26   36.58
   34.87   35.53   35.59   38.73   35.91   35.68    36.9   35.83   36.93   34.27
   35.81   33.19   33.86   27.98   23.81   21.89   25.35   22.89   22.33   27.84
    27.7   22.72   27.25   27.69   25.95   25.46   26.73   26.54   29.26   28.08
   31.13   30.74   32.19   31.47   33.18   31.75   33.37   32.24   32.24   34.18
   33.45   34.54   33.58   34.86   34.16   35.13   34.49   35.64   36.36   38.95
  -964.4  -188.4   955.6  1035.6  1059.6  1083.6    1130    1346    1378    1506
    1538    1554    2674    2722  2780.5  2916.5  2972.5  3020.5  3052.5  3148.5
  3862.7  4006.7  4078.7    4401    4449    4497    4545  4546.5 4785.21  4785.3
 5159.29  5159.4  5200.4    5214    5230    5262    5278    5342  5472.2  5488.2
  5568.2  5608.2  5656.2  5696.2  5736.2  5768.2  5872.2  5888.2  5952.2  6120.2
  6176.2  6344.2  6496.2  6592.2  6624.2  6640.2  6688.2  6864.2  6928.2  6979.7
   38.66   37.16   37.36   36.66   37.43   35.68   36.53   36.36   37.26   36.58
   34.87   35.53   35.59   38.73   35.92    35.9   36.91    35.9   36.94    35.9
   35.82   35.69   35.67   35.57   35.55   35.54   35.52   35.52   35.54   35.54
    35.4    35.4   35.36   35.35   35.34   35.31    35.3   35.31   35.36   35.37
    35.4   35.42   35.44   35.45   35.47   35.48   35.53   35.53   35.56   35.63
   35.65   35.72   35.78    35.8    35.8    35.8    35.8    35.8   36.37   38.95
   38.55   37.05   37.25   36.55   37.32   35.57   36.42   36.25   37.15   36.47
   34.76   35.42   35.48   38.62    35.8   35.57   36.79   35.72   36.82   34.16
    35.7   33.08   33.75   27.87    23.7   21.78   25.24   22.78   22.22   27.73
   27.59   22.61   27.14   27.58   25.84   25.35   26.62   26.43   29.15   27.97
   31.02   30.63   32.08   31.36   33.07   31.64   33.26   32.13   32.13   34.07
   33.34   34.43   33.47   34.75   34.05   35.02   34.38   35.53   36.25   38.84
Pier Skew, UpSta & Num, DnSta & Num=  ,4799.5, 2 ,4799.5, 2 , 0 , 0 , 0 ,,
       1       1
   19.91   28.85
       1       1
    19.8   28.74
Pier Skew, UpSta & Num, DnSta & Num=  ,4815.5, 2 ,4815.5, 2 , 0 , 0 , 0 ,,
       1       1
   15.58   28.87
       1       1
   15.47   28.76
Pier Skew, UpSta & Num, DnSta & Num=  ,4830.8, 2 ,4830.8, 2 , 0 , 0 , 0 ,,
       1       1
   12.23   28.88
       1       1
   12.12   28.77
Pier Skew, UpSta & Num, DnSta & Num=  ,4843.5, 2 ,4843.5, 2 , 0 , 0 , 0 ,,
       1       1
   11.92   28.89
       1       1
   11.81   28.78
Pier Skew, UpSta & Num, DnSta & Num=  ,4860.6, 2 ,4860.6, 2 , 0 , 0 , 0 ,,
       1       1
   10.48   28.91
       1       1
   10.37    28.8
Pier Skew, UpSta & Num, DnSta & Num=  ,4873.7, 2 ,4873.7, 2 , 0 , 0 , 0 ,,
       1       1
   10.04   28.92
       1       1
    9.93   28.81
Pier Skew, UpSta & Num, DnSta & Num=  ,4894.4, 2 ,4894.4, 2 , 0 , 0 , 0 ,,
       1       1
    9.58   28.94
       1       1
    9.47   28.83
Pier Skew, UpSta & Num, DnSta & Num=  ,4905.5, 2 ,4905.5, 2 , 0 , 0 , 0 ,,
       4       4
    8.84   28.95
       4       4
    8.73   28.84
Pier Skew, UpSta & Num, DnSta & Num=  ,4954.7, 2 ,4954.7, 2 , 0 , 0 , 0 ,,
       4       4
    -.23   28.94
       4       4
    -.34   28.83
Pier Skew, UpSta & Num, DnSta & Num=  ,5007.3, 2 ,5007.3, 2 , 0 , 0 , 0 ,,
       4       4
   -7.75   28.92
       4       4
   -7.86   28.81
Pier Skew, UpSta & Num, DnSta & Num=  ,5053.6, 2 ,5053.6, 2 , 0 , 0 , 0 ,,
       4       4
    6.05   28.87
       4       4
    5.94   28.76
Pier Skew, UpSta & Num, DnSta & Num=  ,5070.5, 2 ,5070.5, 2 , 0 , 0 , 0 ,,
       1       1
   10.01   28.84
       1       1
     9.9   28.73
Pier Skew, UpSta & Num, DnSta & Num=  ,5085.6, 2 ,5085.6, 2 , 0 , 0 , 0 ,,
       1       1
   11.58   28.81
       1       1
   11.47    28.7
Pier Skew, UpSta & Num, DnSta & Num=  ,5100.7, 2 ,5100.7, 2 , 0 , 0 , 0 ,,
       1       1
   12.13   28.78
       1       1
   12.02   28.67
Pier Skew, UpSta & Num, DnSta & Num=  ,5115.4, 2 ,5115.4, 2 , 0 , 0 , 0 ,,
       1       1
   13.41   28.75
       1       1
    13.3   28.64
Pier Skew, UpSta & Num, DnSta & Num=  ,5129.9, 2 ,5129.9, 2 , 0 , 0 , 0 ,,
       1       1
   17.84   28.73
       1       1
   17.73   28.62
Pier Skew, UpSta & Num, DnSta & Num=  ,5144.3, 2 ,5144.3, 2 , 0 , 0 , 0 ,,
       1       1
   19.87   28.71
       1       1
   19.76    28.6
BR Coef= 1 , 1 , 0 ,1.25, 0 ,,,0.8,0,2,0,
WSPro=,,,, 1 ,,,, 0 ,,,, 0 ,,,,-1 ,-1 ,-1 , 0 , 0 , 0 , 0 , 0
BR U #Sta/Elev= 183
  -964.4   38.66  -188.4   37.16  -124.4   37.75   -47.4   37.67   379.6   37.23
   595.6   37.38   723.6    37.1   795.6   36.97   851.6   36.88   955.6   37.36
  1003.6   37.03  1035.6   36.66  1059.6   37.43  1083.6   35.68    1130   36.53
    1290   36.54    1346   36.36    1362   36.84    1378   37.26    1410   37.08
    1434    36.7    1458   36.26    1474   36.98    1506   36.58    1538   34.87
    1554   35.53    1930   35.52    1954   34.97    2042   35.71    2610   35.88
    2674   35.59    2722   38.73    2738   38.35  2749.2   37.59    2770   36.17
  2780.5   35.91  2836.5   35.87  2916.5   35.68  2972.5    36.9  3020.5   35.83
  3036.5    36.6  3052.5   36.93  3092.5   35.98  3116.5    35.4  3148.5   34.27
  3228.5   34.88  3348.5   35.27  3359.2   35.27  3444.5   35.23  3862.7   35.81
  3894.7   35.03  3950.7   34.63  4006.7   33.19  4078.7   33.86  4094.7   33.09
    4289   30.02    4401   27.98    4417      27    4433   25.31    4449   23.81
    4473   22.86    4497   21.89    4521   23.25    4545   25.35  4546.5   22.89
  4610.5   23.21  4613.7   23.19  4678.8   22.88  4783.8   22.37 4785.21   22.33
  4785.3   22.33  4785.4   22.33  4799.5   21.98  4800.1   20.69  4815.5   16.68
  4826.9   14.35  4830.8   13.24  4843.3   12.96  4843.5   12.96  4860.6   11.49
  4873.7   11.25  4874.8   10.79  4894.4    10.6  4905.4   10.19  4905.5   10.19
  4919.2     7.8  4954.7    1.59  4954.8    1.08  4999.2   -6.13  5007.3   -6.75
  5007.5   -6.78    5026   -6.46  5032.2   -3.98  5045.2    1.23  5053.1    8.42
  5053.6    8.42  5070.5   11.09  5073.8   11.24  5085.6   12.64  5100.7   13.15
  5106.5   15.46  5115.5   14.33  5124.5   17.25  5129.9      19  5139.1   20.43
  5144.3   20.92  5159.2   22.69 5159.29    22.7  5159.4   22.72  5176.4   24.74
  5200.4   27.25    5214   27.69    5230   25.95    5246   26.04    5262   25.46
    5278   26.73  5287.5   26.84    5294   26.92    5310   27.02    5326   26.93
    5342   26.54    5390   27.43    5406   28.29    5430   28.76    5446   28.66
    5462   28.89  5472.2   29.26  5488.2   28.08  5512.2   29.39  5518.4   29.53
  5528.2   29.75  5544.2   29.89  5568.2   31.13  5584.2   31.35  5608.2   30.74
  5624.2   31.64  5656.2   32.19  5672.2   31.38  5696.2   31.47  5720.2   32.18
  5736.2   33.18  5752.2   32.62  5768.2   31.75  5800.2   32.54  5816.2   32.36
  5872.2   33.37  5888.2   32.24  5920.2    32.3  5952.2   32.24  6008.2   33.08
  6088.2   33.79  6104.2   33.55  6120.2   34.18  6152.2   33.61  6176.2   33.45
  6200.2   33.68  6216.2   34.06  6240.2   33.66  6288.2    34.3  6328.2   33.91
  6344.2   34.54  6376.2    33.9  6392.2   33.91  6416.2   34.13  6448.2   33.99
  6472.2   34.01  6496.2   33.58  6528.2   33.77  6552.9   34.06  6560.2   34.14
  6576.2   34.67  6592.2   34.86  6624.2   34.16  6640.2   35.13  6664.2   34.52
  6688.2   34.49  6784.2   34.94  6864.2   35.64  6904.2   36.53  6928.2   36.36
  6944.2   37.48  6949.6    37.7  6979.7   38.95
BR U #Mann= 5
  -964.4      .2   -47.4      .1  4905.4    .035  5053.1      .1  5518.4     .08
BR U Banks=4905.4,5053.1
BR D #Sta/Elev= 183
  -964.4   38.55  -188.4   37.05  -124.4   37.64   -47.4   37.56   379.6   37.12
   595.6   37.27   723.6   36.99   795.6   36.86   851.6   36.77   955.6   37.25
  1003.6   36.92  1035.6   36.55  1059.6   37.32  1083.6   35.57    1130   36.42
    1290   36.43    1346   36.25    1362   36.73    1378   37.15    1410   36.97
    1434   36.59    1458   36.15    1474   36.87    1506   36.47    1538   34.76
    1554   35.42    1930   35.41    1954   34.86    2042    35.6    2610   35.77
    2674   35.48    2722   38.62    2738   38.24  2749.2   37.48    2770   36.06
  2780.5    35.8  2836.5   35.76  2916.5   35.57  2972.5   36.79  3020.5   35.72
  3036.5   36.49  3052.5   36.82  3092.5   35.87  3116.5   35.29  3148.5   34.16
  3228.5   34.77  3348.5   35.16  3359.2   35.16  3444.5   35.12  3862.7    35.7
  3894.7   34.92  3950.7   34.52  4006.7   33.08  4078.7   33.75  4094.7   32.98
    4289   29.91    4401   27.87    4417   26.89    4433    25.2    4449    23.7
    4473   22.75    4497   21.78    4521   23.14    4545   25.24  4546.5   22.78
  4610.5    23.1  4613.7   23.08  4678.8   22.77  4783.8   22.26 4785.21   22.22
  4785.3   22.22  4785.4   22.22  4799.5   21.87  4800.1   20.58  4815.5   16.57
  4826.9   14.24  4830.8   13.13  4843.3   12.85  4843.5   12.85  4860.6   11.38
  4873.7   11.14  4874.8   10.68  4894.4   10.49  4905.4   10.08  4905.5   10.08
  4919.2    7.69  4954.7    1.48  4954.8     .97  4999.2   -6.24  5007.3   -6.86
  5007.5   -6.89    5026   -6.57  5032.2   -4.09  5045.2    1.12  5053.1    8.31
  5053.6    8.31  5070.5   10.98  5073.8   11.13  5085.6   12.53  5100.7   13.04
  5106.5   15.35  5115.5   14.22  5124.5   17.14  5129.9   18.89  5139.1   20.32
  5144.3   20.81  5159.2   22.58 5159.29   22.59  5159.4   22.61  5176.4   24.63
  5200.4   27.14    5214   27.58    5230   25.84    5246   25.93    5262   25.35
    5278   26.62  5287.5   26.73    5294   26.81    5310   26.91    5326   26.82
    5342   26.43    5390   27.32    5406   28.18    5430   28.65    5446   28.55
    5462   28.78  5472.2   29.15  5488.2   27.97  5512.2   29.28  5518.4   29.42
  5528.2   29.64  5544.2   29.78  5568.2   31.02  5584.2   31.24  5608.2   30.63
  5624.2   31.53  5656.2   32.08  5672.2   31.27  5696.2   31.36  5720.2   32.07
  5736.2   33.07  5752.2   32.51  5768.2   31.64  5800.2   32.43  5816.2   32.25
  5872.2   33.26  5888.2   32.13  5920.2   32.19  5952.2   32.13  6008.2   32.97
  6088.2   33.68  6104.2   33.44  6120.2   34.07  6152.2    33.5  6176.2   33.34
  6200.2   33.57  6216.2   33.95  6240.2   33.55  6288.2   34.19  6328.2    33.8
  6344.2   34.43  6376.2   33.79  6392.2    33.8  6416.2   34.02  6448.2   33.88
  6472.2    33.9  6496.2   33.47  6528.2   33.66  6552.9   33.95  6560.2   34.03
  6576.2   34.56  6592.2   34.75  6624.2   34.05  6640.2   35.02  6664.2   34.41
  6688.2   34.38  6784.2   34.83  6864.2   35.53  6904.2   36.42  6928.2   36.25
  6944.2   37.37  6949.6   37.59  6979.7   38.84
BR D #Mann= 5
  -964.4      .2   -47.4      .1  4905.4    .035  5053.1      .1  5518.4     .08
BR D Banks=4905.4,5053.1
BC Design=,, 0 ,, 0 ,,,,,,
BC HTab HWMax=38.91
BC Use User HTab Curves=0
BC User HTab FreeFlow(D)= 0

Type RM Length L Ch R = 1 ,57937.2 ,40.1,40.1,40.1
BEGIN DESCRIPTION:
Downstream Section of Bridge/Culvert/Weir
END DESCRIPTION:
XS GIS Cut Line= 6
      3169000.55     13869382.95       3165591.3      13867580.4
      3164405.74     13866946.68      3163956.43     13866702.66
      3163476.14     13866466.38       3161979.7     13865666.55
#Sta/Elev= 30
  -964.4   38.33   -47.4   37.34    1954   34.64    2674   35.26    2722    38.4
  2780.5   35.58  3052.5    36.6  3148.5   33.94  3862.7   35.48    4401   27.65
    4497   21.56    4545   25.02  4546.5   22.56  4783.8   22.04  4799.5   21.65
  4830.8   12.91  4905.4    9.86  5007.5   -7.11    5026   -6.79  5045.2      .9
  5053.1    8.09  5106.5   15.13  5115.5      14  5139.1    20.1  5200.4   26.92
    5262   25.13  5518.4    29.2  5736.2   32.85  6784.2   34.61  6979.7   38.62
#Mann= 5 , 1 , 0
  -964.4      .2       0   -47.4      .1       0  4905.4    .035       0
  5053.1      .1       0  5518.4     .08       0
#XS Ineff= 2 , 0
       0    4775    34.6    5169       0    34.7
Permanent Ineff=
       F       F
Bank Sta=4905.4,5053.1
XS Rating Curve= 0 ,0
Exp/Cntr=0.5,0.3

Type RM Length L Ch R = 1 ,57897.1 ,72,72,72
BEGIN DESCRIPTION:
Upstream Section of Bridge/Culvert/Weir
END DESCRIPTION:
XS GIS Cut Line= 5
      3169165.26     13869433.77      3164903.01     13867163.38
       3164233.1     13866794.81      3163501.04     13866415.22
      3161987.41     13865623.15
#Sta/Elev= 30
 -1133.7   37.72  -115.5   36.47  1186.3      35  1274.3   38.01  1826.3   34.66
  4003.8   34.89  4333.7    28.1  4668.3   30.23  4778.9   22.38  4798.5   17.45
  4813.1   19.42  4847.6   12.49  4915.2   12.52    4917     6.4  4943.1    8.15
  4965.4   -2.61  5000.7   -7.99  5028.1   -7.97    5062   10.97  5096.4   14.84
  5131.5   13.28  5162.5   19.79  5169.3   24.03  5169.7   29.64  5747.4   26.57
  5827.4   29.75  5859.4   27.43  6335.3   32.39  6982.3   38.27  6993.1   38.73
#Mann= 6 , 1 , 0
 -1133.7      .2       0  -115.5      .1       0  4915.2    .035       0
  5096.4      .1       0  6335.3     .08       0  6982.3      .2       0
#XS Ineff= 2 , 0
       0    4723    34.6    5221       0    34.7
Permanent Ineff=
       F       F
Bank Sta=4915.2,5096.4
XS Rating Curve= 0 ,0
Exp/Cntr=0.5,0.3
